HEC-RAS study REEDSCK.prj: REEDSCK

--- REEDSCK.g01 (geometry) --- (continued)

Type RM Length L Ch R = 1 ,52233   ,115.3,118.1,120.1
XS GIS Cut Line= 4
2431702.22125367625793.5776354532431896.23788515 625607.83455173
2432007.01037634625381.473374097 2431850.4840301  625087.6854627
#Sta/Elev= 30
       0 2264.21   37.25 2265.07    61.7 2264.12    89.3  2259.6   109.8 2254.83
   139.2  2246.1     155 2243.38   200.5 2240.89     283 2239.33     313 2234.86
   323.1 2234.19     332 2234.69   340.6 2232.98   345.9 2231.86   357.9 2231.03
   371.62232.964   385.4 2236.03   394.3 2236.99   443.3 2235.04   486.5 2238.56
   546.4 2241.57   591.5 2248.17   650.4 2255.33   673.1  2257.2   704.8    2258
   738.6 2257.52   765.2 2258.81   781.9 2261.55   818.1 2271.75   853.5 2279.99
#Mann= 4 ,-1 , 0
       0    .055       0   37.25     .05       0   340.6    .045       0
   371.6     .05       0
#XS Ineff= 2 , 0
                          397.86         2237.09
Permanent Ineff=
       F       F
Bank Sta=340.6,371.6
XS Rating Curve= 0 ,0
Exp/Cntr(USF)=0,0
Exp/Cntr=0.5,0.3

Type RM Length L Ch R = 1 ,52115   ,54.9,57.3,56.8
XS GIS Cut Line= 4
2431723.88515283625880.1052489052431973.82263528625665.873121087
2432095.91191242625508.0784893072431903.56371164625075.007091137
#Sta/Elev= 30
       0 2256.41    11.4 2254.53   23.972254.142   73.572252.261   127.7 2251.36
  189.922245.745  209.212243.703     225 2241.67   296.9 2237.35  306.272236.023
   315.3 2233.55   330.7 2231.53  379.162229.373     424 2228.57   437.5 2227.03
   448.4 2228.54   454.6  2230.1   488.8 2230.32   508.8 2234.28   543.1  2235.4
   578.1 2238.89     635 2239.59   656.9 2238.52   709.3 2242.12     727 2243.95
   788.2 2253.06   846.9 2256.62   921.4 2256.71   942.7 2258.66  1002.6 2266.59
#Mann= 10 ,-1 , 0
       0     .06       0   23.97    .055       0   73.57     .05       0
  189.92     .06       0  209.21     .05       0  306.27     .06       0
  379.16     .05       0     424    .045       0   448.4     .06       0
   788.2     .05       0
#XS Ineff= 2 , 0
             409    2227     463            2227
Permanent Ineff=
       F       F
Bank Sta=424,448.4
XS Rating Curve= 0 ,0
Exp/Cntr(USF)=0,0
Exp/Cntr=0.5,0.3

Type RM Length L Ch R = 1 ,52057   ,288.2,288.8,286.9
XS GIS Cut Line= 4
2431873.61728517626017.1677392832432009.52798992625679.694548688
 2432170.7779786625531.1142019762432543.95652383625245.471364885
#Sta/Elev= 30
       0 2243.29    32.6 2241.26      58 2240.72    67.1 2238.56      78 2239.11
    97.3 2243.04   127.5  2245.1     224 2243.93  262.122240.499  312.572233.683
   338.8 2230.22   363.8 2228.77   387.2 2225.79     4212225.436   430.7 2223.59
   436.2 2223.44   451.22225.443   463.4 2227.73   478.5 2226.99   512.3 2228.17
   523.8 2230.72  538.842231.726   586.1 2233.07   609.8 2234.75   678.7 2246.82
   715.1  2250.5   769.4 2258.22   819.8 2263.87   900.4  2275.7    1053 2295.45
#Mann= 6 ,-1 , 0
       0     .06       0  262.12    .055       0  312.57     .06       0
     421    .045       0   451.2     .06       0  538.84     .05       0
#XS Ineff= 2 , 0
                          463.65         2227.76
Permanent Ineff=
       F       F
Bank Sta=421,451.2
XS Rating Curve= 0 ,0
Exp/Cntr(USF)=0,0
Exp/Cntr=0.5,0.3

Type RM Length L Ch R = 1 ,51769   ,297.1,299,299.9
XS GIS Cut Line= 4
2432040.62620202626066.6945215212432123.55476763625899.685604673
2432269.83154307625664.7213354532432617.67080437625294.998147122
#Sta/Elev= 30
       0 2259.64      40 2249.45    84.6 2236.01      98 2232.94   103.7 2232.85
   124.8 2235.29   138.2 2235.94   159.6 2235.21   189.4 2232.97   195.2 2230.94
   220.52215.448   225.1 2213.63   229.8 2213.44   235.8 2213.78   241.5 2215.44
   250.3 2219.16   260.6 2220.43   338.2 2220.48   366.6  2221.5   383.9 2219.56
   432.4 2226.91   451.3 2226.94   509.7 2229.18   531.7 2230.81   553.6 2234.03
   609.5 2245.82   721.4 2260.52   832.3 2272.66   934.9 2288.88   970.9 2293.48
#Mann= 3 ,-1 , 0
       0     .05       0   220.5    .045       0   241.5     .05       0
#XS Ineff= 2 , 0
                          364.49          2221.8
Permanent Ineff=
       F       F
Bank Sta=220.5,241.5
XS Rating Curve= 0 ,0
Exp/Cntr(USF)=0,0
Exp/Cntr=0.3,0.1

Type RM Length L Ch R = 1 ,51470   ,306.7,309.9,311.9
XS GIS Cut Line= 4
2432224.91190337626215.2748682332432340.09046671626087.426662922
2432479.45652836625919.2659604422432849.17971669625585.248126747
#Sta/Elev= 30
       0 2258.15   48.47 2245.82    74.5 2238.78    86.7 2234.06   113.6 2221.98
   129.7 2216.78   140.5 2215.39   151.7 2214.89   229.9 2212.38   235.1 2211.43
   245.72207.935   255.9 2205.89   262.4 2206.19   268.42207.955   276.5 2212.21
   281.9 2212.92   295.3 2212.29     339 2213.07     358 2212.57   387.4 2215.26
   429.9 2216.49   450.7 2217.96   516.3 2226.19   564.1 2230.98   641.7  2241.2
   718.8 2252.94  767.272261.374  873.332281.221  885.542283.478   888.7 2284.01
#Mann= 7 ,-1 , 0
       0    .055       0   48.47     .05       0   245.7    .045       0
   268.4     .05       0  767.27      .1       0  873.33     .05       0
  885.54      .1       0
Bank Sta=245.7,268.4
XS Rating Curve= 0 ,0
Exp/Cntr(USF)=0,0
Exp/Cntr=0.3,0.1

Type RM Length L Ch R = 1 ,51160   ,309.6,309.8,309.2
XS GIS Cut Line= 4
2432371.18867882626428.3552104182432469.09045766626346.578430445
2432750.12615221626142.7123733272433040.37613184625923.873102976
#Sta/Elev= 30
       0 2261.04    9.512258.012    40.5 2247.96    82.8 2232.69     103 2223.84
   131.4 2208.72   147.5 2202.89   154.3 2201.97     184 2202.35   198.8 2201.34
   230.7  2200.4   254.5 2198.48   258.1 2198.56   264.72200.386   274.6  2202.7
   297.6 2204.29   322.3 2204.96   337.2 2206.29   416.2 2206.45     436 2207.27
   452.2    2209   487.7 2214.98     521 2218.78   545.7 2222.34   645.9  2238.5
   683.6 2244.97     695 2247.74   760.2 2259.49   801.1 2267.99   838.3 2274.71
#Mann= 4 ,-1 , 0
       0    .055       0    9.51     .05       0   230.7    .045       0
   264.7     .05       0
Bank Sta=230.7,264.7
XS Rating Curve= 0 ,0
Exp/Cntr(USF)=0,0
Exp/Cntr=0.3,0.1

Type RM Length L Ch R = 1 ,50850   ,298.6,297.6,296.7
XS GIS Cut Line= 4
2432572.75116467626655.2569802042432654.52794464626584.998056565
2432800.80472008626458.3016368872433170.52790842626165.748085996
#Sta/Elev= 30
       0 2241.47    13.2 2238.06    58.4 2220.09    81.7 2211.92   103.8 2206.53
   118.7 2201.05   129.4 2199.33   145.1 2195.11   163.3 2193.44   196.6 2195.15
   207.7 2194.88   214.9 2194.24   221.3 2192.08   227.1 2190.27   231.4 2189.98
   243.82192.062   251.2 2194.16   266.9 2195.91   306.8 2196.26   329.3 2199.12
   403.5 2199.48   427.6 2200.71   493.1  2207.5   524.4 2209.55   579.2  2211.4
   661.4 2218.49     700 2224.74   712.9 2228.38   737.4 2238.01   772.8 2254.14
#Mann= 3 ,-1 , 0
       0     .05       0   221.3    .045       0   243.8     .05       0
Bank Sta=221.3,243.8
XS Rating Curve= 0 ,0
Exp/Cntr(USF)=0,0
Exp/Cntr=0.3,0.1

Type RM Length L Ch R = 1 ,50552   ,347,347.8,348
XS GIS Cut Line= 4
2432774.31365052626871.7926792892432883.73328569 626764.67661538
2433046.13506001626624.158768101 2433366.3314661626347.730216078
#Sta/Elev= 30
       0 2218.04    12.7 2212.11      23 2208.11    34.2 2204.23    46.2 2201.08
    57.5 2196.14    81.3 2196.92    88.6 2195.38    98.5 2194.54   112.6 2191.52
   139.22190.508   167.9 2188.73   178.52185.284   193.4 2183.48   199.4 2183.63
   207.6    2185   220.6  2185.4   250.1 2190.82   267.1 2192.03   320.9 2190.97
     374 2191.22   416.2 2189.12   479.7 2190.09   496.8 2191.23   506.1 2192.76
   532.5 2198.88   627.6 2210.72   701.6  2223.2   749.2 2233.22   790.9 2248.69
#Mann= 4 ,-1 , 0
       0     .06       0   139.2     .05       0   178.5    .045       0
   207.6     .05       0
Bank Sta=178.5,207.6
XS Rating Curve= 0 ,0
Exp/Cntr(USF)=0,0
Exp/Cntr=0.3,0.1

Type RM Length L Ch R = 1 ,50205   ,463.2,462,460.4
XS GIS Cut Line= 4
2432972.42077947627111.3640910422433058.80470197627044.560524303
2433420.46539087626794.6230418492433716.47429866626568.873057697
#Sta/Elev= 30
       0 2226.05    13.9 2218.71   23.442212.221    27.7 2209.94    36.2 2208.03
    59.6 2195.58    78.8 2187.82    87.5 2183.08   107.5 2183.15   118.9 2180.95
  135.722180.528   196.6 2181.41   216.1 2179.57   226.92175.934   231.1 2174.17
   235.5 2173.68   245.5 2176.12   259.9 2178.94   285.7 2178.34   309.1 2176.07
   337.7 2174.78   372.5 2175.59   397.9  2177.7   449.6  2187.8   548.4 2200.02
   624.5  2212.2   746.3  2236.1   787.1 2242.08  914.112266.773   921.1 2268.25
#Mann= 6 ,-1 , 0
       0      .1       0   23.44     .06       0  135.72     .05       0
   226.9    .045       0   245.5     .05       0  914.11      .1       0
#XS Ineff= 2 , 0
                          287.09         2176.65
Permanent Ineff=
       F       F
Bank Sta=226.9,245.5
XS Rating Curve= 0 ,0
Exp/Cntr(USF)=0,0
Exp/Cntr=0.3,0.1

Type RM Length L Ch R = 1 ,49743   ,279.7,275.3,252.1
XS GIS Cut Line= 4
2433264.97433036627499.515849508 2433349.0546816627426.953354602
 2433741.8135826627054.9265950042433992.90285069626831.480182119
#Sta/Elev= 30
       0 2213.79    39.3 2200.56    69.8 2188.74    78.3 2184.64    92.5  2174.3
   113.4 2173.71   126.4 2169.14   149.1  2168.6  172.732169.403   202.8 2169.79
   262.3 2168.06   271.82166.046   278.7  2163.9   282.1 2163.81   293.22166.034
   306.2 2168.61   343.8 2170.25   399.9 2169.25     495 2169.18   528.2 2170.21
   548.6 2172.47   593.3 2179.37   649.9 2185.37   680.1 2192.21   707.32200.098
   743.4 2210.62   797.2 2229.43   859.6 2248.61   883.5 2254.28   988.2 2274.09
#Mann= 5 ,-1 , 0
       0     .06       0  172.73     .05       0   271.8    .045       0
   293.2     .05       0   707.3      .1       0
#XS Ineff= 2 , 0
          192.43  2169.9  359.78            2170
Permanent Ineff=
       F       F
Bank Sta=271.8,293.2
XS Rating Curve= 0 ,0
Exp/Cntr(USF)=0,0
Exp/Cntr=0.3,0.1

Type RM Length L Ch R = 1 ,49467   ,351.2,354.9,348.5
XS GIS Cut Line= 4
2433522.20281139627694.1993232972433669.07781139627528.574323311
2433708.66114473627406.6993233112434176.71670029626901.317378864
#Sta/Elev= 30
       0 2172.75     5.6 2171.81    22.6 2171.86    57.9 2170.24   87.482167.747
   148.8 2162.98   227.3 2160.72   265.6 2158.59   273.6 2157.29   281.2 2156.92
   289.9 2158.75     297 2159.38   392.9 2161.79   411.4 2161.31     431 2162.14
   458.4 2161.54   481.1 2161.84     551 2165.12   567.3 2166.98   577.3 2168.92
   605.7 2176.66   670.5 2192.15   709.1 2202.43   752.7 2217.34  773.642221.321
   834.5 2233.57  899.652249.107  934.082257.379 1025.662278.504  1038.3 2281.39
#Mann= 8 ,-1 , 0
       0     .06       0   87.48     .05       0   265.6    .045       0
   289.9     .05       0  773.64      .1       0  899.65     .05       0
  934.08      .1       0 1025.66     .05       0
#XS Ineff= 2 , 0
                          392.58         2161.97
Permanent Ineff=
       F       F
Bank Sta=265.6,289.9
XS Rating Curve= 0 ,0
Exp/Cntr(USF)=0,0
Exp/Cntr=0.3,0.1

Type RM Length L Ch R = 1 ,49112   ,366.8,373.2,384
XS GIS Cut Line= 4
2433602.44752095 627953.319389082433916.88499888627699.926549725
2434091.95641516627482.239065007 2434485.0960848627158.411927246
#Sta/Elev= 30
       0 2197.93   17.712194.534      23 2193.02    50.3 2191.14   108.3 2181.99
  148.84 2177.19   231.6 2170.72   297.1 2162.69   419.6 2155.09   425.7 2154.21
   436.22149.748   445.7 2147.25   454.5 2150.13   461.6 2152.14   534.5 2151.49
   574.6  2149.5     590 2153.34   610.5 2156.37   646.4 2163.98   676.2 2168.19
  700.142174.051  761.152190.392   869.4 2225.57   943.6 2247.96   988.8 2259.49
  1059.6 2280.38  1153.2 2304.56  1162.1 2307.87  1173.5 2309.52  1192.5 2316.33
#Mann= 7 ,-1 , 0
       0     .05       0   17.71     .06       0  148.84     .05       0
   436.2    .045       0   454.5     .05       0  700.14      .1       0
  761.15      .1       0
#XS Ineff= 2 , 0
                          477.36         2151.58
Permanent Ineff=
       F       F
Bank Sta=436.2,454.5
XS Rating Curve= 0 ,0
Exp/Cntr(USF)=0,0
Exp/Cntr=0.3,0.1

Type RM Length L Ch R = 1 ,48739   ,271,272.8,276.4
XS GIS Cut Line= 4
2433813.61612018628044.7654805442434112.22721033627931.008874773
2434319.20103472627867.8107604562434756.84797636627564.459811734
#Sta/Elev= 30
       0 2186.55      44 2179.98   157.3 2167.02   169.7 2163.67   188.3  2154.8
   198.1 2153.53   215.2 2147.15   347.3 2145.47   397.5 2141.68   403.52139.391
     410 2137.17   414.2 2137.07   421.4 2139.35   430.9 2141.39   460.2 2140.43
   485.3 2141.44   520.3 2152.54   540.3 2156.16   579.4 2160.57     657 2173.78
   783.5 2200.68   812.8 2208.51   827.4 2210.37  870.592221.678   929.6 2235.92
     954  2243.2   968.6  2245.7  1002.6  2255.7  1036.1 2263.51  1068.5 2273.57
#Mann= 4 ,-1 , 0
       0     .05       0   403.5    .045       0   421.4     .05       0
  870.59      .1       0
Bank Sta=403.5,421.4
XS Rating Curve= 0 ,0
Exp/Cntr(USF)=0,0
Exp/Cntr=0.3,0.1

Type RM Length L Ch R = 1 ,48466   ,103.1,98,92.2
XS GIS Cut Line= 4
2433960.55173597628254.8992106482434074.30834174628188.541190616
 2434406.0984419628147.4624163092434802.66660924627845.691420445
#Sta/Elev= 30
       0 2172.28    33.8 2169.95    55.6 2166.63    81.3 2164.87    85.9  2163.6
     127  2145.1   140.7 2140.41   152.3 2138.39   237.6 2137.58   278.42132.866
   293.4 2130.68   303.52132.886   313.5 2135.48   321.6 2136.42   424.1    2137
   638.7 2142.21   698.2 2148.44   732.3 2155.42  761.762159.055   795.1 2166.93
   803.6 2167.89     818 2167.53   823.7 2169.15   874.32196.305   897.9 2207.96
   929.3 2221.08   934.3 2223.01  941.73 2223.98   954.4 2229.52   964.3 2232.47
#Mann= 6 ,-1 , 0
       0     .05       0   278.4    .045       0   303.5     .05       0
  761.76      .1       0   874.3     .05       0  941.73      .1       0
#XS Ineff= 2 , 0
          212.92 2138.05
Permanent Ineff=
       F       F
Bank Sta=278.4,303.5
XS Rating Curve= 0 ,0
Exp/Cntr(USF)=0,0
Exp/Cntr=0.5,0.3

Type RM Length L Ch R = 1 ,48368   ,29.2,29.4,29.6
XS GIS Cut Line= 4
2434055.06855217628389.9348557592434225.90188551628284.726522416
2434417.56855217628165.9765224312434813.48869106627876.393189102
#Sta/Elev= 30
       0 2165.08    54.3 2161.48    65.4 2159.89    82.1 2154.28    97.3 2145.76
   107.7 2144.38   121.8 2138.27   156.1 2133.72   173.4  2132.1   211.3 2131.93
   228.7 2130.82   248.7 2128.93   266.5 2129.42   278.1    2131   296.5 2132.19
     356 2136.72   385.1 2136.01   576.2 2140.08   618.1 2142.55   669.6 2147.95
   702.4 2154.78   724.9 2158.28  750.552165.138   789.8 2173.66     807 2180.73
  820.99 2188.02     847 2200.61   888.4 2217.13   903.3 2219.91   916.6 2225.13
#Mann= 7 ,-1 , 0
       0     .05       0   156.1      .1       0   228.7    .045       0
   278.1      .1       0   296.5     .05       0  750.55      .1       0
  820.99     .05       0
#XS Ineff= 2 , 0
           224.9 2129.28  280.38         2129.37
Permanent Ineff=
       F       F
Bank Sta=228.7,278.1
XS Rating Curve= 0 ,0
Exp/Cntr(USF)=0,0
Exp/Cntr=0.5,0.3

Type RM Length L Ch R = 1 ,48339   ,129.7,127.9,125.7
XS GIS Cut Line= 4
2434086.05813551628434.7265224312434254.80813551628300.351522431
2434372.51646885628228.4765224312434820.43313554627899.309855744
#Sta/Elev= 30
       0 2163.77    46.9 2159.51    57.1  2156.7   102.8  2140.1   108.9 2138.79
   139.9  2135.7   154.3  2132.4     211 2131.64   234.4 2130.01   256.9 2127.11
   267.2 2128.32   272.8 2130.04   298.2 2133.15   341.9 2135.04   390.1 2135.11
   425.9 2136.32   435.8 2135.82   450.7 2136.84   540.1 2138.29   599.5 2140.31
   618.8 2141.76   664.2  2146.5   725.5 2158.18  795.522180.021  810.172185.316
   847.8 2199.91   876.4 2209.38   887.5 2213.78   897.5 2214.74   909.5 2219.04
#Mann= 5 ,-1 , 0
       0     .05       0   234.4    .045       0   272.8     .05       0
  795.52      .1       0  810.17     .05       0
Bank Sta=234.4,272.8
XS Rating Curve= 0 ,0
Exp/Cntr(USF)=0,0
Exp/Cntr=0.5,0.3

Type RM Length L Ch R = 1 ,48211   ,376.5,377.9,378.1
XS GIS Cut Line= 4
2434159.62579606628534.5508665022434230.72367467628493.472092196
2434432.95764049628322.8371835392434887.98406357627900.989770472
#Sta/Elev= 30
       0 2157.35    37.2 2155.31    51.8 2153.29    63.5 2149.52    92.5 2136.83
   103.8  2132.8   113.5 2130.69   244.4 2128.81   271.12126.969     281 2125.09
   291.2 2125.42   298.8 2126.97     311 2130.58   322.9 2132.06   480.1 2132.79
   507.3 2134.56   571.5 2135.86   611.2  2137.9   643.7 2140.83   680.4 2146.57
   713.1  2155.2   744.2 2164.69   787.9 2180.96   861.9 2199.07   872.8 2203.07
   883.7 2208.37  900.542210.217   911.5 2211.52   933.8 2221.58   967.2 2234.83
#Mann= 4 ,-1 , 0
       0     .05       0   271.1    .045       0   298.8     .05       0
  900.54    .055       0
#XS Ineff= 2 , 0
          148.02 2130.77
Permanent Ineff=
       F       F
Bank Sta=271.1,298.8
XS Rating Curve= 0 ,0
Exp/Cntr(USF)=0,0
Exp/Cntr=0.3,0.1

Type RM Length L Ch R = 1 ,47833   ,321.2,321.7,321.5
XS GIS Cut Line= 4
2434357.11990331628831.5820037932434576.73335056628678.326576573
2434843.74538355628495.0520450542435107.59751082628278.598503517
#Sta/Elev= 30
       0 2155.36    21.8 2150.31   39.212144.446      85 2127.12    90.7 2125.63
   109.3 2123.16   226.4 2122.14   280.3 2122.95   289.6 2122.28   299.4 2119.64
   325.9 2117.38   338.2  2115.1     343 2115.73   347.52117.389   352.7 2119.51
   357.6 2120.34   521.3 2121.32   542.5 2122.52   565.2 2124.37   619.5 2131.37
   661.3 2137.55  694.022144.373   738.9 2154.28   775.8  2164.4  802.782172.522
     818 2177.73   828.4 2179.82   850.5  2187.5   886.6  2201.4   932.9 2216.69
#Mann= 6 ,-1 , 0
       0     .06       0   39.21     .05       0   325.9    .045       0
   347.5     .05       0  694.02    .055       0  802.78      .1       0
#XS Ineff= 2 , 0
                           402.9         2120.84
Permanent Ineff=
       F       F
Bank Sta=325.9,347.5
XS Rating Curve= 0 ,0
Exp/Cntr(USF)=0,0
Exp/Cntr=0.3,0.1

Type RM Length L Ch R = 1 ,47512   ,372.8,374.7,375.6
XS GIS Cut Line= 4
2434486.67603766629003.7968653072434807.40646782628871.080825241
 2434924.3229793628768.3838894752435279.81237234628476.092610759
#Sta/Elev= 30
       0 2153.99   21.112150.928    99.6 2144.67     111 2142.62   138.5 2135.45
   160.2 2130.75   199.2 2128.87   298.8 2120.66   329.1 2117.55   367.5  2115.1
   401.1  2108.7   409.1 2107.07   415.4 2106.72   430.32108.712   451.6 2110.05
   468.6 2114.75   471.5 2114.91   599.3 2116.18   613.5 2116.92   636.2 2119.66
   644.8 2121.29   684.5 2133.09   738.9  2146.3  776.592157.236     820  2171.5
   840.8 2179.02   851.5 2181.15   873.5  2188.6     909 2203.75   962.9 2224.92
#Mann= 5 ,-1 , 0
       0     .06       0   21.11     .05       0   401.1    .045       0
   430.3     .05       0  776.59    .055       0
Bank Sta=401.1,430.3
XS Rating Curve= 0 ,0
Exp/Cntr(USF)=0,0
Exp/Cntr=0.3,0.1

Type RM Length L Ch R = 1 ,47137   ,369,369.1,375.8
XS GIS Cut Line= 4
2434816.88618496 629283.44852116 2435003.3206222629176.011726821
 2435322.4710995  628932.69898672435606.86261393628690.966199437
#Sta/Elev= 30
       0 2148.28    62.2 2143.76   130.6 2132.74   189.2 2129.97   221.3 2126.93
   230.2 2124.81   243.4 2119.93   249.7 2116.34   263.2 2106.14   270.32101.728
   274.8 2100.21     283 2099.54   294.72101.736     305 2105.73     310 2106.62
   335.8 2106.02   410.6 2107.08   513.9 2106.44   541.4 2107.47   561.5 2110.91
  592.322120.276   640.7 2134.75   663.4 2143.56   736.6 2174.39   767.5 2185.37
   779.6    2188     786 2190.75  823.692202.682   947.6 2248.02   989.7 2266.45
#Mann= 5 ,-1 , 0
       0     .05       0   270.3    .045       0   294.7     .05       0
  592.32    .055       0  823.69      .1       0
#XS Ineff= 2 , 0
                          479.94         2109.43
Permanent Ineff=
       F       F
Bank Sta=270.3,294.7
XS Rating Curve= 0 ,0
Exp/Cntr(USF)=0,0
Exp/Cntr=0.3,0.1

Type RM Length L Ch R = 1 ,46768   ,138.2,137,146.6
XS GIS Cut Line= 4
2435085.05003363629583.2618233112435264.21670029629440.206267744
2435400.32781142 629330.484045522435869.77225584628974.928489983
#Sta/Elev= 30
       0 2140.51    78.3 2127.56   140.9  2115.5   166.5 2111.55   177.9 2111.34
   191.6 2109.66   220.6 2100.38   249.1 2098.95     276 2094.93   286.1 2092.93
     295 2094.97   304.4 2098.68   314.2 2099.59   439.8 2098.31   472.4 2098.61
   487.4 2099.62   499.8  2102.5   542.6 2119.57  589.862134.694     663 2160.32
   708.2 2174.28   748.2 2185.28   768.2 2192.47  789.372201.351  814.68 2211.62
   863.8 2232.38  927.092260.851     944 2268.73   979.2 2283.16     993 2289.95
#Mann= 7 ,-1 , 0
       0     .05       0     276    .045       0     295     .05       0
  589.86      .1       0  789.37    .055       0  814.68      .1       0
  927.09      .1       0
#XS Ineff= 2 , 0
                          329.49         2099.75
Permanent Ineff=
       F       F
Bank Sta=276,295
XS Rating Curve= 0 ,0
Exp/Cntr(USF)=0,0
Exp/Cntr=0.3,0.1

Type RM Length L Ch R = 1 ,46631   ,312.1,338,284.4
XS GIS Cut Line= 4
2435185.01520086 629695.816217082435360.38996809629539.400884145
2435548.40435818629378.2456926362435916.53337408629063.835073908
#Sta/Elev= 30
       0 2132.11      16 2128.13    38.7 2123.68    69.9 2118.22   123.7 2109.91
   163.1 2106.95   211.4 2106.34     235 2103.71   253.9 2102.35   266.5 2099.61
   282.62093.401   290.9 2090.92   293.8 2090.83   307.32093.392   441.3 2095.59
   469.9 2101.42  512.582115.044   545.6 2125.54  592.282142.837   605.8  2147.8
   628.82155.231   662.6 2165.91   697.2 2175.88   736.3 2188.66   793.1 2205.38
   827.6 2217.22   838.9 2220.62  861.252228.588   906.5 2244.21   966.7 2262.13
#Mann= 7 ,-1 , 0
       0     .05       0   282.6    .045       0   307.3     .05       0
  512.58      .1       0  592.28     .05       0   628.8      .1       0
  861.25      .1       0
Bank Sta=282.6,307.3
XS Rating Curve= 0 ,0
Exp/Cntr(USF)=0,0
Exp/Cntr=0.3,0.1

Type RM Length L Ch R = 1 ,46293   ,319.1,326.6,326.6
XS GIS Cut Line= 4
2435312.99138235629850.651597157  2435472.566621 629725.83532138
2435783.81733402629498.3221098392436049.24941415629275.548756871
#Sta/Elev= 30
       0 2118.42    23.9 2118.36    83.5 2113.08   149.5 2105.95   205.3 2102.53
   220.2 2100.76   254.8 2091.17   263.5 2090.01   314.3 2089.71   406.6 2090.54
   449.6 2089.36   475.3 2086.39   486.8 2085.99     499 2084.91   502.6 2084.98
   505.8 2086.25   507.5  2087.3   517.4  2097.2   532.9 2110.21   547.2 2119.05
   557.1 2126.34   566.8 2131.88  601.022148.752  621.542157.831   691.2 2184.35
  716.642194.898  809.95 2234.48   856.7 2254.41   894.8 2267.84   934.7 2280.84
#Mann= 7 ,-1 , 0
       0     .05       0   486.8    .045       0   505.8      .1       0
  601.02     .12       0  621.54      .1       0  716.64     .12       0
  809.95      .1       0
#XS Ineff= 2 , 0
          351.79 2090.81
Permanent Ineff=
       F       F
Bank Sta=486.8,505.8
XS Rating Curve= 0 ,0
Exp/Cntr(USF)=0,0
Exp/Cntr=0.3,0.1

Type RM Length L Ch R = 1 ,45966   ,262.6,262.5,259.3
XS GIS Cut Line= 4
2435480.46638529630075.0049029832435700.07983255629923.329428621
2435899.15389264629814.3126814242436256.22323854629534.661025571
#Sta/Elev= 30
       0 2121.97    50.6 2114.48   104.9 2102.89     157 2097.17   197.3 2090.68
   269.9  2088.8   283.6  2087.4   301.1 2083.69   313.4 2082.25   343.1 2080.97
   384.4 2082.43   410.6 2080.95   420.4 2079.38   434.1 2081.08  438.492082.368
   443.2  2084.4   460.7 2095.98   531.9 2136.69   544.8  2145.4  605.752182.281
   625.4 2193.56     661 2212.49   696.6 2229.96   737.2 2246.95  774.462260.407
  805.452270.731     855 2286.99  887.862295.608   929.1  2309.6   947.4 2313.49
#Mann= 8 ,-1 , 0
       0     .05       0   410.6    .045       0   434.1     .05       0
  438.49      .1       0  605.75      .1       0  774.46     .12       0
  805.45      .1       0  887.86     .12       0
Bank Sta=410.6,434.1
XS Rating Curve= 0 ,0
Exp/Cntr(USF)=0,0
Exp/Cntr=0.3,0.1

Type RM Length L Ch R = 1 ,45704   ,230.2,236.3,230.9
XS GIS Cut Line= 4
2435670.06072824630218.7806130542435867.55483549630136.623064442
2436031.86993271630026.0263643872436371.55979717629757.434378539
#Sta/Elev= 30
       0 2117.63    22.4 2114.26      83 2112.44   126.4 2108.58     174 2106.39
   208.5 2103.45   227.4 2099.58   251.5 2089.79   263.5 2083.86   275.6  2081.4
   283.82077.597   288.6 2075.89   292.4  2075.6   306.8 2077.48   317.3 2077.99
     350  2076.4  356.912076.972   362.4 2078.64   373.1 2083.63   407.7 2103.71
  582.112213.822  593.01 2220.08   634.9 2241.26   678.4  2258.4   707.2 2268.47
   731.8 2275.68  791.062294.928  809.492300.181   823.6  2306.9     845 2308.02
#Mann= 8 ,-1 , 0
       0     .05       0   283.8    .045       0   306.8     .05       0
  356.91      .1       0  582.11     .12       0  593.01      .1       0
  791.06     .12       0  809.49      .1       0
Bank Sta=283.8,306.8
XS Rating Curve= 0 ,0
Exp/Cntr(USF)=0,0
Exp/Cntr=0.5,0.3

Type RM Length L Ch R = 1 ,45467   ,84.6,84.9,96.6
XS GIS Cut Line= 4
2435722.27185039630293.3812471472436014.42428041630216.435428147
2436187.95230395630242.5579263132436609.64406006630339.584348073
#Sta/Elev= 30
       0 2106.85     .442106.859    25.3 2108.08      46 2107.76  128.03 2102.73
   174.2 2103.01   207.3 2100.68   276.8 2092.54  299.792086.887   322.1 2082.34
  362.232076.244   383.3 2073.95   391.32071.557   399.5 2069.15   403.6 2069.31
   409.1 2071.55   419.7 2075.83   431.9 2077.99   476.4  2092.3  509.142101.795
   533.8 2107.87   562.6 2113.92   603.6 2121.62  647.472128.057   710.3    2138
  723.63 2139.41     776 2146.83   858.1 2160.72     895 2164.68   910.3 2165.67
#Mann= 10 ,-1 , 0
       0     .05       0     .44     .06       0  128.03     .05       0
  299.79      .1       0  362.23     .06       0   391.3    .045       0
   409.1     .06       0  509.14      .1       0  647.47     .06       0
  723.63      .1       0
#XS Ineff= 2 , 0
             378    2081     422            2081
Permanent Ineff=
       F       F
Bank Sta=391.3,409.1
XS Rating Curve= 0 ,0
Exp/Cntr(USF)=0,0
Exp/Cntr=0.5,0.3

Type RM Length L Ch R = 1 ,45382   ,236,236.5,218.1
XS GIS Cut Line= 4
2435797.98072418630370.3715780552436074.13284765630304.132386276
2436210.34301666630306.9312253652436584.45450826630412.354164393
#Sta/Elev= 30
       0 2120.02   37.452116.678   41.652116.359    70.7 2113.69     135 2109.47
   165.3 2106.54   202.6 2104.24   235.8 2101.12   255.7 2098.44   276.4  2094.3
   296.6  2087.3   312.6 2078.51   316.6 2077.58   328.6 2076.02   349.5 2068.52
   352.6 2067.51   360.6  2066.9   383.9 2067.38   391.72068.511   404.9 2072.09
   420.2 2078.03   475.6 2089.92   499.6  2093.6     521 2097.46   620.1 2111.45
   653.4 2115.52   661.7 2116.15   753.1  2127.4   785.4 2131.86   808.9 2134.43
#Mann= 5 ,-1 , 0
       0     .06       0   37.45     .05       0   41.65     .06       0
   349.5    .045       0   391.7     .06       0
Bank Sta=349.5,391.7
XS Rating Curve= 0 ,0
Exp/Cntr(USF)=0,0
Exp/Cntr=0.5,0.3

Type RM Length L Ch R = 1 ,45146   ,192.7,188.2,184.3
XS GIS Cut Line= 4
2436062.93749129630595.2116515572436253.25854936630490.721658892
2436383.87104019630439.4096089232436572.32620554630425.415413476
#Sta/Elev= 30
       0 2121.61     8.9 2119.16    17.3 2117.45    40.8  2111.5    68.2 2106.54
    82.6 2103.55    91.4 2101.41   103.2 2097.78   117.9 2094.91   132.1 2092.79
   154.9 2090.66   203.4 2087.39   209.7 2086.57   231.6 2080.77   235.9 2080.01
   244.5 2077.14   253.1 2073.61   270.3 2064.71   273.62063.805   282.9 2062.06
   295.3 2061.67   304.82063.797  323.312066.003     339  2067.5   357.4 2073.45
   416.5 2088.44   468.9 2103.35   492.7 2110.73   532.4 2121.86   546.4 2126.39
#Mann= 4 ,-1 , 0
       0     .05       0   273.6    .045       0   304.8     .05       0
  323.31     .06       0
Bank Sta=273.6,304.8
XS Rating Curve= 0 ,0
Exp/Cntr(USF)=0,0
Exp/Cntr=0.3,0.1

Type RM Length L Ch R = 1 ,44958   ,185.1,182.3,180.8
XS GIS Cut Line= 4
2436233.66667574630742.617176923 2436434.2501438630587.748080652
2436534.07540465630500.0511225232436584.45450825630434.744877107
#Sta/Elev= 30
       0 2104.93    23.4 2097.98    31.9 2094.75    41.8 2092.76    67.1 2086.53
    92.3 2082.58   117.5 2080.88   128.9 2081.07   195.9 2079.69   220.2 2078.47
   243.9 2079.11   260.8 2077.78   265.7 2076.34   285.5 2064.63  300.592060.214
   301.82059.893   309.3 2058.85     318 2058.74   327.4 2057.94   333.5 2058.76
   337.32059.885   351.7 2064.58   356.4  2066.8   376.2  2076.9   392.8 2087.15
   410.4 2096.55   433.2 2107.81   448.4  2114.6  458.112119.496   468.8 2125.41
#Mann= 5 ,-1 , 0
       0     .05       0  300.59      .1       0   301.8    .045       0
   337.3      .1       0  458.11     .06       0
Bank Sta=301.8,337.3
XS Rating Curve= 0 ,0
Exp/Cntr(USF)=0,0
Exp/Cntr=0.3,0.1

Type RM Length L Ch R = 1 ,44775   ,249.5,256.1,260.9
XS GIS Cut Line= 4
2436261.65506663 630790.197441442436543.40486828630708.098161489
2436669.35262729630610.138793366 2436833.5511872630504.715854338
#Sta/Elev= 30
       0    2102    30.3 2090.29    59.5 2083.52    84.5 2079.77   109.5 2077.69
     181 2075.39   205.3 2073.92   222.9  2071.7   255.3 2070.28   307.8 2071.58
   312.9 2071.26   333.8  2068.3   373.7  2057.9   379.4 2057.43   390.8 2058.32
   407.82055.401   419.3 2052.56   424.4 2053.52   426.92055.353   430.7 2058.84
   439.6 2069.46     453 2083.55     459 2089.26   473.8 2101.39   481.2 2106.81
     507 2124.04   530.7 2138.43   540.3 2143.01   568.8  2151.9   648.2 2171.05
#Mann= 3 ,-1 , 0
       0     .05       0   407.8    .045       0   426.9      .1       0
Bank Sta=407.8,426.9
XS Rating Curve= 0 ,0
Exp/Cntr(USF)=0,0
Exp/Cntr=0.3,0.1

Type RM Length L Ch R = 1 ,44519   ,293.5,290.6,290.2
XS GIS Cut Line= 4
2436238.33140755630892.8215413792436581.65566917630868.564935939
2436779.44029814630859.2354723082436934.30939441630845.241276862
#Sta/Elev= 30
       0 2120.58    28.4 2109.17    54.6 2099.79    80.6 2092.96    96.7 2089.76
   200.7 2075.92   271.9 2069.32   301.2 2064.68   329.2 2064.14   345.3 2062.82
   377.3 2055.47   429.4  2054.7   461.4 2052.75   481.4 2052.49   485.4 2051.88
   490.42049.853   497.4  2047.7   501.4 2047.64   505.4 2048.22   508.62049.852
   525.5 2066.26   541.8 2080.11   567.6 2099.49  582.922110.256     594  2118.3
   617.8 2133.36   641.9 2144.97   653.9 2149.63  682.482162.426   697.7 2168.81
#Mann= 5 ,-1 , 0
       0     .05       0   490.4    .045       0   508.6     .05       0
  582.92      .1       0  682.48     .12       0
Bank Sta=490.4,508.6
XS Rating Curve= 0 ,0
Exp/Cntr(USF)=0,0
Exp/Cntr=0.3,0.1

Type RM Length L Ch R = 1 ,44229   ,228.7,232.7,234.1
XS GIS Cut Line= 4
2436282.53821993631157.8858084862436551.28820106631151.486999411
2436781.64532775631148.9274757812436969.77031454631134.850095817
#Sta/Elev= 30
       0 2120.83    60.2 2107.04   132.2 2088.64   188.3 2076.49   198.5 2073.81
   216.3 2070.02   240.3  2065.9   256.3    2064   292.3 2053.82   308.3 2047.58
   312.3 2046.78   316.4 2046.44   397.1 2047.53   408.3  2047.1   415.3 2045.38
   420.3 2043.66   424.3 2043.32   437.6 2043.51   446.9 2045.42   456.3 2048.75
   472.3 2055.88   488.3 2060.77   517.1 2068.38   524.4 2070.82   548.4 2080.77
   560.5 2084.49   567.6 2087.82  584.332098.092   628.3 2119.54   687.8  2151.1
#Mann= 4 ,-1 , 0
       0     .05       0   415.3    .045       0   446.9     .05       0
  584.33      .1       0
Bank Sta=415.3,446.9
XS Rating Curve= 0 ,0
Exp/Cntr(USF)=0,0
Exp/Cntr=0.3,0.1

Type RM Length L Ch R = 1 ,43996   ,320.8,314.8,275
XS GIS Cut Line= 4
2436411.79416323631371.6060315782436579.44296099631367.766746133
2436741.97271148631372.8857933932436968.49055272631330.653653501
#Sta/Elev= 30
       0 2101.49      31 2095.09      47 2091.17      67 2085.72   89.122078.658
     135  2061.9     143 2060.82     167 2054.52     175 2051.81     191 2044.48
     195 2043.34     211 2041.53   220.5 2041.34     231 2039.47     235 2039.33
   248.12041.594   259.3 2042.33   295.1  2042.9   307.1 2043.85   315.1 2045.49
   339.2 2052.19   378.8 2056.23   392.1 2058.27   420.6  2069.8   449.3 2083.74
  490.17 2105.21   504.2  2112.3   526.4 2124.64   546.7  2134.6   560.7 2143.02
#Mann= 5 ,-1 , 0
       0      .1       0   89.12     .05       0   220.5    .045       0
   248.1     .05       0  490.17      .1       0
Bank Sta=220.5,248.1
XS Rating Curve= 0 ,0
Exp/Cntr(USF)=0,0
Exp/Cntr=0.3,0.1

Type RM Length L Ch R = 1 ,43681   ,268.3,278.8,284.4
XS GIS Cut Line= 4
2436488.57987213631674.9095817152436711.25842792631663.391725381
2436859.71079845631599.4036346352437029.91911984631530.296496629
#Sta/Elev= 30
       0 2068.89    26.2 2062.81    58.2 2058.83   154.4    2050   194.4 2042.69
   213.5 2041.24   239.8 2040.47   257.3 2039.27   261.6 2038.63   270.3  2036.2
   292.1 2034.67   298.52033.702   305.2 2032.11   313.9 2031.21   317.3 2031.96
   321.12033.722   326.5 2036.18   329.5 2036.64   347.8    2037   353.1 2037.73
   357.4 2038.95   366.2 2042.98   378.2 2049.67     386 2054.78   448.3 2100.42
  466.552112.058   508.8 2135.22   521.7 2142.93   537.8 2151.65   568.3  2166.9
#Mann= 4 ,-1 , 0
       0     .05       0   298.5    .045       0   321.1     .05       0
  466.55      .1       0
Bank Sta=298.5,321.1
XS Rating Curve= 0 ,0
Exp/Cntr(USF)=0,0
Exp/Cntr=0.3,0.1

Type RM Length L Ch R = 1 ,43402   ,227.2,225.4,223.4
XS GIS Cut Line= 4
2436451.46677949631879.6714721032436724.05604607631855.355997619
2436916.02031831631877.1119484732437127.18101777631820.802428616
#Sta/Elev= 30
       0 2064.57    35.4 2057.47    63.5 2053.73   111.7 2050.03   167.9 2047.09
   208.1 2045.62   232.3 2045.78   244.2 2045.37   256.3 2043.66   286.5 2036.28
   300.5 2033.91   324.7 2031.73     381 2031.14   391.72028.144   401.2 2026.65
   409.5 2026.37   417.3 2026.58   424.82028.131  435.092030.901     442 2033.97
   452.9 2041.73   463.7 2050.06   486.2 2064.87   519.9 2083.46   531.8 2089.27
   556.6 2100.26   578.8 2109.01   614.3 2124.05  635.742132.567   685.4 2152.17
#Mann= 5 ,-1 , 0
       0     .05       0   391.7    .045       0   424.8     .05       0
  435.09      .1       0  635.74     .12       0
Bank Sta=391.7,424.8
XS Rating Curve= 0 ,0
Exp/Cntr(USF)=0,0
Exp/Cntr=0.3,0.1

Type RM Length L Ch R = 1 ,43177   ,271.9,263.7,257.2
XS GIS Cut Line= 4
2436450.18701768632102.3500278992436708.69890429 632094.67145701
2436912.18103287 632089.552409752437188.60958489  632016.6059863
#Sta/Elev= 30
       0 2069.75    64.6 2062.65   120.6 2054.71   196.6 2046.57   208.7 2044.03
   248.7 2042.66   256.7 2041.78   264.7  2039.5   287.7  2030.2   299.4 2027.46
   312.7 2026.24   336.7 2025.86   367.7 2026.45   386.42022.769   392.7  2021.2
   400.7 2020.65   404.7 2021.29   407.62022.754   416.7 2029.57   420.7 2031.83
   444.7 2042.62   469.4 2052.46   485.5 2058.01   502.1 2062.83   571.2 2078.45
   613.7 2090.81   639.9 2097.69  668.982104.366   707.8  2115.1   748.1 2127.63
#Mann= 5 ,-1 , 0
       0     .05       0   386.4    .045       0   407.6     .05       0
   469.4      .1       0  668.98     .12       0
Bank Sta=386.4,407.6
XS Rating Curve= 0 ,0
Exp/Cntr(USF)=0,0
Exp/Cntr=0.3,0.1

Type RM Length L Ch R = 1 ,42913   ,408.9,404.5,399.4
XS GIS Cut Line= 4
2436619.11557725632582.2607084962436820.03818219632426.129767075
2437004.32388354632269.9988256552437207.80601211632084.433362491
#Sta/Elev= 30
       0 2098.67    14.7 2093.92    44.9 2082.37   88.182063.165     116 2052.38
   155.4 2040.47   173.2 2036.53   213.1 2030.41   235.9 2025.74   284.2 2021.12
   341.9 2021.06   358.5 2019.31   387.1 2020.59   411.9 2019.49   414.8 2019.12
   422.12016.507   440.3 2014.03   445.1 2015.14   447.4 2016.47   457.2 2023.17
   482.2  2036.2   499.9 2043.37  527.63 2053.14   553.7 2057.95   596.7 2069.66
   631.2 2077.47  704.192098.097   721.2 2103.14   760.4 2113.24   771.4 2117.05
#Mann= 6 ,-1 , 0
       0      .1       0   88.18     .05       0   422.1    .045       0
   447.4     .05       0  527.63      .1       0  704.19     .12       0
Bank Sta=422.1,447.4
XS Rating Curve= 0 ,0
Exp/Cntr(USF)=0,0
Exp/Cntr=0.3,0.1

Type RM Length L Ch R = 1 ,42509   ,373.5,376.5,380.5
XS GIS Cut Line= 4
2437100.30601966632780.6237898092437183.49053763632668.004750096
2437287.15124464632504.1952377862437467.59766054632240.564303911
#Sta/Elev= 30
       0 2045.58    41.9 2043.12      63 2040.65    74.5    2038   121.5 2024.53
     132 2022.56   151.9 2017.22   166.4 2012.44   174.5 2011.38   178.52010.129
   183.8 2008.66   193.4 2008.03   204.1 2008.65     2102010.115   217.1 2011.72
   236.2 2010.71   254.9 2010.65   273.9 2015.15   288.1 2020.46  333.492045.999
  335.852047.049   354.8 2054.16   397.8 2067.79     413 2071.96   420.8 2073.18
     441 2077.91  479.872089.906   504.3 2097.26   611.7 2136.19   653.3 2149.94
#Mann= 6 ,-1 , 0
       0     .05       0   178.5    .045       0     210     .05       0
  333.49      .1       0  335.85     .12       0  479.87      .1       0
Bank Sta=178.5,210
XS Rating Curve= 0 ,0
Exp/Cntr(USF)=0,0
Exp/Cntr=0.3,0.1

Type RM Length L Ch R = 1 ,42132   ,240,246.7,247
XS GIS Cut Line= 4
2437297.38933916632839.4928332952437481.67504051   632848.451166
2437613.49050745632738.3916499162437856.64525228632458.123812448
#Sta/Elev= 30
       0 2040.97    73.6 2035.21   133.5 2026.02   165.6 2022.75   193.2 2017.67
   226.1 2004.68   243.72003.338   253.6 2001.28   268.7 2003.02   282.9 2003.44
   299.3 2001.87   305.5 2002.97   314.2 2007.27   345.4 2027.21   364.2  2037.1
  375.332041.985   393.6 2048.97   413.1 2054.75   429.7 2060.85   474.1 2078.95
  489.652083.596  504.692087.866   535.2 2098.56   575.1 2115.18   602.3 2123.26
     629 2134.17   654.5 2147.78   668.7 2152.13   678.6 2156.25   727.3  2182.8
#Mann= 6 ,-1 , 0
       0     .05       0   243.7    .045       0   268.7     .05       0
  375.33      .1       0  489.65     .12       0  504.69      .1       0
Bank Sta=243.7,268.7
XS Rating Curve= 0 ,0
Exp/Cntr(USF)=0,0
Exp/Cntr=0.3,0.1

Type RM Length L Ch R = 1 ,41886   ,268,266.5,261.8
XS GIS Cut Line= 4
2437420.24647339633057.052341832  2437575.097653633005.861869235
2437692.83573997632980.2666329372438033.25238274632793.421407958
#Sta/Elev= 30
       0  2037.5    11.1 2034.72    40.5 2025.74    86.9 2018.09     108 2016.08
   132.7 2012.57   145.9 2010.12   166.8 2004.79   183.2 2002.25   191.4 1998.57
     1991997.707   215.9 1995.18   228.3 1997.72   244.6 1999.11   256.1 2002.61
   265.1 2003.65   269.2  2004.8   281.4 2011.92   299.4 2019.38   317.7 2026.04
   340.5 2032.83  362.512038.246  414.872051.816   467.9 2064.19   536.7  2079.9
   577.7 2092.61   598.3 2100.64     628 2113.35   638.9 2119.14   671.9 2134.77
#Mann= 6 ,-1 , 0
       0      .1       0     199    .045       0   228.3      .1       0
  362.51      .1       0  414.87     .12       0   467.9      .1       0
Bank Sta=199,228.3
XS Rating Curve= 0 ,0
Exp/Cntr(USF)=0,0
Exp/Cntr=0.3,0.1

Type RM Length L Ch R = 1 ,41619   ,280.3,279.4,280
XS GIS Cut Line= 5
2437482.95480232633309.165419372 2437584.0559857633278.451135814
2437672.35955093633250.2963758862437749.14525983633210.623759623
2438081.88333171633054.492818203
#Sta/Elev= 30
       0 2050.99    12.3 2046.24    20.9 2042.31    83.4 2009.47   104.3 2000.51
   116.9 1996.79   129.5 1995.52   199.7 1996.23   205.3  1995.2   214.5 1991.97
     228  1991.3   238.3 1991.73   246.1 1990.88   250.6 1991.05   255.1 1992.01
     259 1992.72   268.6 1993.07   273.1 1994.19   277.6 1996.31   286.5 2001.85
   294.8  2005.7   303.8 2008.56   366.1 2017.48   383.7 2022.98   410.3 2029.66
   453.6 2042.13   499.3 2052.89   560.5 2065.91   638.3 2086.28   652.3 2090.36
#Mann= 3 ,-1 , 0
       0      .1       0   238.3    .045       0   255.1      .1       0
#XS Ineff= 2 , 0
          199.43 1996.58
Permanent Ineff=
       F       F
Bank Sta=238.3,255.1
XS Rating Curve= 0 ,0
Exp/Cntr(USF)=0,0
Exp/Cntr=0.3,0.1

Type RM Length L Ch R = 1 ,41340   ,387.3,399.5,391.7
XS GIS Cut Line= 4
2437557.18098759633581.7546859512437681.31788364633529.284451539
2437837.44882506633457.6177899032438135.63332793633265.653517665
#Sta/Elev= 30
       0 2074.49     6.4 2071.74    61.4 2043.58   101.1    2015   116.3 2002.86
   127.6 1995.85   131.6    1994   140.7 1990.87   145.1 1990.02   189.2 1988.92
     201 1986.52   215.6 1984.43   224.4 1986.58   233.2 1986.79   250.8 1991.25
   265.2 1991.79   281.6 1993.65  315.321999.383   326.4 2001.13   360.4 2004.16
   398.5 2006.31  423.672008.521   468.6 2014.39   503.4 2018.15   517.4 2020.72
     541 2026.68   555.5 2027.03   617.3 2042.39  640.372047.473   661.2  2053.5
#Mann= 6 ,-1 , 0
       0      .1       0     201    .045       0   224.4      .1       0
  315.32      .1       0  423.67     .05       0  640.37      .1       0
Bank Sta=201,224.4
XS Rating Curve= 0 ,0
Exp/Cntr(USF)=0,0
Exp/Cntr=0.3,0.1

Type RM Length L Ch R = 1 ,40940   ,194.3,259.1,261.4
XS GIS Cut Line= 4
2437740.18692712633943.9272795742437934.71072299633813.391574452
2437980.78214833633745.5641982612438206.02022776633574.076115062
#Sta/Elev= 30
       0  2051.5    36.8 2029.12    80.8 2009.32    97.7 2002.71   126.5 1994.65
   133.1 1992.05   142.8 1989.86   157.2 1984.29   166.9 1982.47   187.1 1981.19
   205.4 1980.59   237.3  1981.3   245.61980.254   251.8 1978.98   261.5 1978.09
   274.5 1980.25   280.8 1981.09   290.5 1984.02   295.3 1984.77   348.1 1985.99
   384.1  1988.7   402.3 1991.12   413.8 1993.32   424.3 1996.59   439.4 1999.69
   481.1  2005.7     532 2014.71  554.912020.676   585.2 2029.31   599.3 2031.51
#Mann= 4 ,-1 , 0
       0      .1       0   245.6    .045       0   274.5     .05       0
  554.91      .1       0
Bank Sta=245.6,274.5
XS Rating Curve= 0 ,0
Exp/Cntr(USF)=0,0
Exp/Cntr=0.3,0.1

Type RM Length L Ch R = 1 ,40681   ,299.1,300.1,300.2
XS GIS Cut Line= 4
2437793.93692335634079.5820319562437930.87143755634027.111797545
2438129.23451886 633932.409423242438349.35355103633830.028478046
#Sta/Elev= 30
       0 2029.29    35.1 2012.98    52.3 2006.23    65.1 2001.87    73.7 1999.58
    97.4  1994.5   137.9 1989.81   146.6 1988.24  153.89 1986.25   159.8 1984.06
   172.41974.632   177.5 1972.17     182 1972.07   195.3 1973.73   198.3 1974.65
   204.1 1977.28   208.6 1978.61   221.7    1980   248.5 1980.81  295.881980.834
     346  1982.1     399 1985.49   407.9 1986.66   434.3 1991.67   447.5 1995.53
  464.052001.069   512.3 2016.48   552.4 2026.89  567.232030.154   609.2 2038.83
#Mann= 7 ,-1 , 0
       0      .1       0  153.89    .055       0   172.4    .045       0
   198.3    .055       0  295.88     .05       0  464.05      .1       0
  567.23     .12       0
Bank Sta=172.4,198.3
XS Rating Curve= 0 ,0
Exp/Cntr(USF)=0,0
Exp/Cntr=0.3,0.1

Type RM Length L Ch R = 1 ,40381   ,344.2,341.7,340.4
XS GIS Cut Line= 4
2437873.28215588634375.2070112042438006.37738463634315.058205902
2438194.50237142634236.9927351922438455.57378167634094.939173735
#Sta/Elev= 30
       0 2035.29    63.1 2012.21   104.1 1994.41   137.7 1982.68   150.8 1980.86
   159.4 1977.71   172.4 1974.92   177.1 1974.45   198.4 1974.91   219.9  1972.3
  226.031970.831   230.61969.583   241.7 1967.65   250.4 1967.96   256.21969.571
   263.4 1973.81   268.9 1975.47   302.4 1974.96   328.11976.773  341.821977.696
   359.1 1979.51   401.6 1987.13  432.681990.981     455 1994.11   486.6 1999.98
   527.6 2010.28   545.8  2015.8   594.8 2028.91  633.222037.334     647 2039.46
#Mann= 8 ,-1 , 0
       0      .1       0  226.03    .055       0   230.6    .045       0
   256.2    .055       0   328.1     .05       0  341.82    .055       0
  432.68     .12       0  633.22      .1       0
#XS Ineff= 2 , 0
          194.29 1975.18
Permanent Ineff=
       F       F
Bank Sta=230.6,256.2
XS Rating Curve= 0 ,0
Exp/Cntr(USF)=0,0
Exp/Cntr=0.3,0.1

Type RM Length L Ch R = 1 ,40039   ,329.7,316.9,303.6
XS GIS Cut Line= 4
2438033.25238274634678.510561341 2438115.1571389634640.117706893
2438278.96665121634562.0522361832438566.91305956 634353.45106035
#Sta/Elev= 30
       0 2031.84    18.9 2025.39    45.8 2013.25    59.1 2004.58    63.5 2000.97
    67.9 1996.31    81.2 1989.23   102.6 1975.69   116.6 1968.79   125.4 1966.66
   175.1 1967.25   178.6 1966.84   183.51964.262   187.5 1961.97   191.9 1961.24
   203.7 1964.28   222.9 1965.88   232.1 1968.27   249.5 1970.98   267.2 1975.98
   279.8 1977.93  324.43 1980.37   408.6 1984.28   474.2 1988.21   493.9 1990.61
   503.2 1992.45   513.7 1995.66  573.252017.919   597.6 2026.37   627.5 2033.26
#Mann= 5 ,-1 , 0
       0      .1       0   183.5    .045       0   203.7      .1       0
  324.43     .05       0  573.25     .12       0
Bank Sta=183.5,203.7
XS Rating Curve= 0 ,0
Exp/Cntr(USF)=0,0
Exp/Cntr=0.3,0.1

Type RM Length L Ch R = 1 ,39722   ,240.4,235.4,236.5
XS GIS Cut Line= 4
2438323.75831473634957.4986369942438364.71069281634898.629593507
2438461.97259074634706.6653212692438659.05591024634492.945098177
#Sta/Elev= 30
       0 2003.11       8 2005.56    32.4 2007.76    42.2 2006.93    47.1 2005.76
    58.6 2000.64    84.9  1984.9    89.4 1981.86   105.8 1968.21   118.81959.163
   120.7 1957.76   125.2 1956.78     1481959.142   156.6 1961.09  186.041962.744
   228.4 1964.38   251.6 1967.03   264.2 1969.42   312.8 1975.59   382.5 1980.42
   400.9 1982.14   417.9 1984.72   434.5 1988.66   459.2 1996.87   482.8 2002.47
   505.3  2013.3  525.032024.429   561.9 2042.63   565.4 2043.54   577.6 2044.15
#Mann= 5 ,-1 , 0
       0      .1       0   118.8    .045       0     148      .1       0
  186.04     .05       0  525.03     .06       0
Bank Sta=118.8,148
XS Rating Curve= 0 ,0
Exp/Cntr(USF)=0,0
Exp/Cntr=0.3,0.1

Type RM Length L Ch R = 1 ,39487   ,213,318.8,327
XS GIS Cut Line= 4
  2438467.091638635050.9212494832438542.59758508635015.087918665
2438662.89519568 634860.236739062438820.30589892634762.974841125
#Sta/Elev= 30
       0 1995.03    37.4 1982.95    74.7 1967.82    98.1 1959.21   103.8  1958.2
   149.7 1957.33  162.571955.678   165.31955.282   188.1 1953.09   194.7 1953.73
     1991955.272   210.5 1957.44   225.7 1957.43   229.2 1957.96   245.9 1964.18
     251 1965.43   272.9 1968.67  294.391973.024   303.8 1975.42   331.2 1984.38
   367.7  2000.5   373.5 2003.67   378.2 2007.03   382.9 2009.36  401.892010.965
   405.5  2013.1   411.1 2017.82   415.8 2020.84   448.8 2033.79   464.7 2040.61
#Mann= 6 ,-1 , 0
       0      .1       0  162.57     .05       0   165.3    .045       0
     199     .05       0  294.39    .055       0  401.89     .06       0
Bank Sta=165.3,199
XS Rating Curve= 0 ,0
Exp/Cntr(USF)=0,0
Exp/Cntr=0.3,0.1

Type RM Length L Ch R = 1 ,39168   ,313.9,255.9,248.5
XS GIS Cut Line= 4
2438509.32377789635224.9688563132438588.66901042 635195.53433457
2438766.55590269635177.6176691612438911.16898778635157.141480122
#Sta/Elev= 30
       0 1985.66    39.9 1976.58    65.5 1969.22    77.4 1964.15    94.8 1955.97
   102.8 1952.95   106.8    1952   110.8 1951.64  125.931951.768   167.5 1952.52
   179.2 1952.16   191.2 1949.87   207.3 1949.71   211.3 1948.81   215.4 1948.58
   219.4 1948.93   222.2 1949.75  225.42 1950.75   239.5 1956.29   251.5 1960.38
   275.7 1967.23   279.8 1968.73   287.8 1972.88     304 1973.37     308 1974.24
   316.1 1981.45   321.6  1985.3   328.2 1988.71   340.4 1993.82   409.5 2031.36
#Mann= 5 ,-1 , 0
       0      .1       0  125.93     .05       0   207.3    .045       0
   222.2     .05       0  225.42     .06       0
Bank Sta=207.3,222.2
XS Rating Curve= 0 ,0
Exp/Cntr(USF)=0,0
Exp/Cntr=0.5,0.3

Type RM Length L Ch R = 1 ,38912   ,91.6,101.4,101.2
XS GIS Cut Line= 4
2438634.74043575635601.2188299012438717.92495372635546.189071859
2438792.15113899635382.3795595492438961.07969856635336.308134211
#Sta/Elev= 30
       0 1970.71    13.2 1969.74    33.2 1966.99    88.3 1956.63   108.9 1951.01
   116.5 1949.69     130 1949.16   145.2 1947.88   156.1 1947.76   169.3 1945.73
   182.4 1945.95   190.21944.748   204.4 1943.06   213.1 1943.85   227.7 1943.66
   234.71944.726   248.3 1949.87   256.8 1950.93   274.6 1952.09   290.6 1951.89
   294.7 1952.96   298.9  1956.2   307.3 1964.99   319.6 1975.26  348.871993.052
   368.9 2004.62     398 2023.16   402.5 2025.79   414.5 2031.58   454.7 2055.46
#Mann= 5 ,-1 , 0
       0      .1       0   108.9     .06       0   190.2    .045       0
   234.7     .06       0  348.87      .1       0
#XS Ineff= 2 , 0
             172  1948.6     252          1948.6
Permanent Ineff=
       F       F
Bank Sta=190.2,234.7
XS Rating Curve= 0 ,0
Exp/Cntr(USF)=0,0
Exp/Cntr=0.5,0.3

Type RM Length L Ch R = 1 ,38811   ,106.9,115.4,123
XS GIS Cut Line= 4
2438682.09162291635649.849778868 2438758.8773318635601.218829901
2438855.44496973635432.1815121152438983.89926678635394.883740806
#Sta/Elev= 30
       01965.715  17.1121964.441  27.9581963.261  48.9991962.184  65.337 1960.33
  72.8131958.803  95.4311952.071 118.8861947.154 127.6811946.151 151.136 1945.17
 195.4531945.809 203.5171944.433 211.5811941.591 219.6451939.334 227.3631938.324
 236.1591938.595  239.091939.689 242.0221941.638 250.1991948.882 259.4131954.894
 265.477 1959.62 277.2041971.214 280.1361973.487 301.4991988.603 322.325 2001.06
 338.985 2011.77 347.3742016.527 363.9772029.246 384.8032041.953 419.3262061.779
#Mann= 6 ,-1 , 0
       0     .05       0  17.112      .1       0 151.136     .06       0
 211.581    .045       0 242.022     .06       0 322.325      .1       0
#XS Ineff= 2 , 0
          163.64 1945.09
Permanent Ineff=
       F       F
Bank Sta=211.581,242.022
XS Rating Curve= 0 ,0
Exp/Cntr(USF)=0,0
Exp/Cntr=0.5,0.3
