HEC-RAS study REEDSCK.prj: REEDSCK

--- REEDSCK.g01 (geometry) --- (continued)

Type RM Length L Ch R = 1 ,38695   ,153.6,154.4,155.2
XS GIS Cut Line= 4
 2438713.2479879635680.4394580542438803.36515944635638.938129057
2438905.33985355635595.065295545 2439039.3298586635534.591930435
#Sta/Elev= 30
       0 1961.41    23.7 1960.44    32.4 1959.53    45.7 1957.88    80.7 1948.69
    94.1 1945.78   102.9 1944.59   111.6 1942.74     129 1942.03   146.4 1942.62
   150.8 1942.21   155.1 1939.86   160.1 1936.36   163.9 1935.18   168.2 1934.94
   172.6 1935.04   178.31936.416   185.6 1939.73   194.3 1941.27   198.7 1943.85
   211.4 1955.71   220.7 1963.75   233.7 1976.03   250.7  1989.9     260 1996.93
   278.7 2009.31   299.5 2025.57   330.3 2047.34     339 2054.92   357.2 2066.13
#Mann= 6 ,-1 , 0
       0     .05       0    32.4      .1       0   150.8     .06       0
   160.1    .045       0   178.3     .06       0   278.7      .1       0
Bank Sta=160.1,178.3
XS Rating Curve= 0 ,0
Exp/Cntr(USF)=0,0
Exp/Cntr=0.3,0.1

Type RM Length L Ch R = 1 ,38541   ,258.9,259.7,260
XS GIS Cut Line= 4
2438758.30657367635815.6152153592438885.18206518635768.185125077
2438984.78525477635732.6125573652439129.44703013635672.139192254
#Sta/Elev= 30
       0 1954.22    17.5 1953.63    25.8 1952.46    53.7 1944.15    64.5  1941.8
    73.1 1940.46    98.7 1939.82   115.8 1940.31   150.2 1939.33   162.7 1938.36
   172.91935.362   179.6 1932.64   184.6 1932.02   187.8  1932.1   190.9 1932.76
   192.3 1933.17   195.4 1935.17   203.4 1942.48   213.6 1950.27   222.5 1958.17
   231.6 1965.37   243.3 1976.54   274.6 1998.29   282.4 2003.02     317 2026.95
   338.7 2041.27   360.2 2054.07   382.1 2064.86   393.8 2072.08     398 2074.05
#Mann= 6 ,-1 , 0
       0     .05       0    25.8      .1       0   150.2     .06       0
   172.9    .045       0   195.4     .06       0   274.6      .1       0
#XS Ineff= 2 , 0
          115.44 1940.33
Permanent Ineff=
       F       F
Bank Sta=172.9,195.4
XS Rating Curve= 0 ,0
Exp/Cntr(USF)=0,0
Exp/Cntr=0.3,0.1

Type RM Length L Ch R = 1 ,38281   ,118.1,119.4,120.7
XS GIS Cut Line= 4
2438790.32188461636070.5519506292438974.11348446636008.892833261
2439072.53092179635979.2490268352439234.97898101 635916.40415721
#Sta/Elev= 30
       0 1946.87      38 1946.06      68 1944.35    72.2 1943.35    93.3 1935.95
    97.5 1935.21   122.8 1935.03     177  1936.5     212 1935.89   219.6 1935.13
   223.8 1932.79   224.8 1931.82   227.9    1929   232.1  1927.7   234.5 1927.65
   240.5 1928.49   245.9 1931.14     253 1934.82   261.4  1940.9   270.1 1946.31
   304.8 1963.39     329 1975.57   341.9  1981.5   354.8 1988.67   372.9 1997.59
   386.3 2004.97   397.6 2010.27     444 2035.41   462.5 2046.17   470.8 2050.41
#Mann= 5 ,-1 , 0
       0     .05       0      38      .1       0   224.8    .045       0
   245.9     .06       0   304.8      .1       0
#XS Ineff= 2 , 0
           178.9 1936.39
Permanent Ineff=
       F       F
Bank Sta=224.8,245.9
XS Rating Curve= 0 ,0
Exp/Cntr(USF)=0,0
Exp/Cntr=0.5,0.3

Type RM Length L Ch R = 1 ,38162   ,34.2,35.4,36.9
XS GIS Cut Line= 4
2438817.44239479636160.6431890732439021.43545035636113.768189073
2439138.62295032636092.9348557592439271.43545035636039.115411296
#Sta/Elev= 30
       0 1941.25    12.6 1938.89    17.8 1937.29    25.9 1933.59    29.2 1932.65
    42.4  1931.1    54.7 1931.15    62.9 1932.35     108    1934  168.85 1934.16
   226.9 1932.75     231 1932.05   237.1  1928.8   243.1 1925.81   247.2 1925.37
   251.3 1925.63   256.8 1928.51   259.4 1930.07   263.5 1931.07   275.6 1931.42
   296.3 1935.01     313 1940.87   328.5 1947.19   339.4 1952.99     350 1958.83
   358.7 1965.17   368.4 1970.71   380.3 1978.73  443.362014.407   471.6 2029.25
#Mann= 6 ,-1 , 0
       0     .05       0  168.85     .06       0   237.1    .045       0
   256.8     .06       0   296.3      .1       0  443.36      .1       0
#XS Ineff= 3 ,-1
   11.65  134.791936.826  141.47  230.09 1932.14     264   471.6    1932
Permanent Ineff=
       F       F       F
Bank Sta=237.1,256.8
XS Rating Curve= 0 ,0
Exp/Cntr(USF)=0,0
Exp/Cntr=0.5,0.3

Type RM Length L Ch R = 1 ,38127   ,42.5,39.8,37.3
XS GIS Cut Line= 4
2438831.33128369636185.8168002072439036.19239479636145.018189088
2439157.72017255636126.7890224312439286.19239476636076.441800207
#Sta/Elev= 30
       0 1940.59     7.6 1940.02    15.6 1938.58    19.8 1937.34      28 1933.79
      32 1932.57    44.3 1930.97    60.6 1930.87      81 1933.49  158.91 1933.88
   174.8 1933.52   195.2  1931.9   219.6    1932   223.6 1931.04   227.6 1929.13
   235.7 1925.74   247.9 1924.84     256 1925.46     260 1926.27   265.8 1929.02
   268.1 1930.05   272.1 1930.65   293.9 1932.43   316.6 1935.18   332.9 1939.85
   341.5  1944.4   350.1 1949.85   380.1 1972.24     422 1997.76   469.8 2024.31
#Mann= 4 ,-1 , 0
       0    .055       0  158.91      .1       0   227.6    .045       0
   265.8      .1       0
#XS Ineff= 2 , 0
          160.03 1938.74
Permanent Ineff=
       F       F
Bank Sta=227.6,265.8
XS Rating Curve= 0 ,0
Exp/Cntr(USF)=0,0
Exp/Cntr=0.5,0.3

Type RM Length L Ch R = 1 ,38087   ,145.1,143.8,142.5
XS GIS Cut Line= 4
2438837.08611462636265.5896075692439020.10132833636198.948198228
2439186.20752773636144.242563696 2439295.6187968636104.456647672
#Sta/Elev= 30
       0 1940.81    12.8 1937.93    27.3 1932.79    34.6 1931.23    86.9  1930.2
   108.2 1931.04   113.1 1932.33     121    1933   189.1 1933.12   212.7 1931.59
   244.4 1930.88   248.1  1930.4  257.59 1925.47   260.7  1924.1   264.9 1923.39
   269.1 1923.73  277.12 1925.36   284.5 1926.91   290.2 1929.27   294.4 1930.04
   340.7 1932.54     345  1933.3   349.2 1934.89   361.8 1941.89     395 1964.89
   417.9 1979.82   433.6 1989.06   455.2 2002.66   463.9 2007.15   486.1 2019.68
#Mann= 4 ,-1 , 0
       0    .055       0   108.2      .1       0  257.59    .045       0
  277.12      .1       0
#XS Ineff= 2 , 0
          120.16 1934.47
Permanent Ineff=
       F       F
Bank Sta=257.59,277.12
XS Rating Curve= 0 ,0
Exp/Cntr(USF)=0,0
Exp/Cntr=0.3,0.1

Type RM Length L Ch R = 1 ,37943   ,102.3,98.7,96.2
XS GIS Cut Line= 4
 2438844.6213734636434.3437714162439114.65111635636320.444969888
2439172.24039802636294.8497335892439330.93086307636187.349741136
#Sta/Elev= 30
       0 1946.25    62.3 1940.66    80.4  1936.3    97.8 1930.23   106.5 1928.41
   162.9 1926.71     176 1927.08  190.871929.182   228.1 1929.58   267.1 1928.23
   301.9 1928.44   315.1 1927.64   321.51924.722   326.4 1922.35   332.6 1921.65
   336.7 1922.66   340.61924.686   346.1 1927.98   351.9 1929.13  398.411929.533
   420.2 1929.69   431.6 1931.86   436.4 1935.12   450.9 1948.28   455.8 1951.95
   478.8 1966.94   494.4 1975.24   507.91983.724   527.8 1996.05   547.8 2007.48
#Mann= 6 ,-1 , 0
       0     .05       0  190.87     .06       0   321.5    .045       0
   340.6     .06       0  398.41     .05       0   507.9      .1       0
#XS Ineff= 2 , 0
           191.9 1931.25
Permanent Ineff=
       F       F
Bank Sta=321.5,340.6
XS Rating Curve= 0 ,0
Exp/Cntr(USF)=0,0
Exp/Cntr=0.3,0.1

Type RM Length L Ch R = 1 ,37845   ,98.1,95.7,94.1
XS GIS Cut Line= 4
2438976.55239597636579.0507483012439178.18045691636413.806698362
2439276.72048669636321.3306704142439370.71251509636224.306641092
#Sta/Elev= 30
       0 1943.35      39 1938.71    50.7 1938.02    84.1 1929.83   106.8 1928.36
   126.7 1927.22   147.6 1927.65   160.8 1926.64   230.4 1927.12   243.3 1926.72
   251.8 1925.53   299.9    1926   305.3 1924.16   308.4 1922.12   311.7 1920.44
   317.6 1920.02   323.4  1920.2   329.2 1922.03   336.7 1924.42   354.7 1926.01
   362.2 1927.96   376.3 1936.67   382.1 1939.56     416 1954.03   443.8 1968.93
   479.2  1989.1   495.2 1997.06   513.7 2004.68   523.5 2010.44   530.9 2015.55
#Mann= 4 ,-1 , 0
       0    .055       0   106.8      .1       0   308.4    .045       0
   329.2      .1       0
#XS Ineff= 2 , 0
          140.89 1929.96
Permanent Ineff=
       F       F
Bank Sta=308.4,329.2
XS Rating Curve= 0 ,0
Exp/Cntr(USF)=0,0
Exp/Cntr=0.3,0.1

Type RM Length L Ch R = 1 ,37749   ,177,175.9,175
XS GIS Cut Line= 4
2439094.17492731636714.6116088842439272.06181959636465.058054974
2439336.04991033636378.0342515592439423.07371375636251.337831882
#Sta/Elev= 30
       0 1954.88    28.5 1949.08    69.9 1943.33   112.1  1933.9     147 1927.24
   171.6 1925.18  204.231925.116   209.6 1924.58   215.8 1923.04   225.6 1922.59
     244 1924.47   289.5  1924.3   304.3 1925.78     330 1924.28     334 1923.43
   338.61921.578   344.3  1919.5   353.8 1918.72   358.8 1918.93     3661921.561
   368.7 1922.54   383.6  1924.6   388.6 1926.71   395.8  1931.8   418.3 1952.01
   431.7  1961.6   461.8 1978.63   520.2 2008.36   539.3 2018.93   568.2 2033.84
#Mann= 4 ,-1 , 0
       0     .05       0  204.23     .06       0   338.6    .045       0
     366      .1       0
#XS Ineff= 2 , 0
          304.45  1925.7
Permanent Ineff=
       F       F
Bank Sta=338.6,366
XS Rating Curve= 0 ,0
Exp/Cntr(USF)=0,0
Exp/Cntr=0.3,0.1

Type RM Length L Ch R = 1 ,37573   ,222.8,224.2,226.1
XS GIS Cut Line= 4
2439266.94277233636787.558032335  2439393.639192636607.111616431
2439474.26418634636480.4151967532439557.44870431636321.724731703
#Sta/Elev= 30
       0 1948.23    31.9 1945.24    55.3 1941.66    95.1 1934.43   135.3 1931.94
   157.2 1928.84   172.6 1929.06  176.271928.474   181.7 1927.23   209.9 1927.02
   270.7 1921.54   305.5 1919.92   310.41918.147   315.6 1915.98     320 1915.59
   328.6 1916.23   332.21918.188   341.8  1926.7   369.2 1953.14   381.4 1964.24
   395.8 1975.43   414.8 1988.76   422.5 1994.89   431.1 2000.35   444.6 2010.04
   489.8 2039.02   507.9 2050.34   516.9 2054.98   535.1 2066.92   549.8 2075.41
#Mann= 4 ,-1 , 0
       0     .05       0  176.27     .06       0   310.4    .045       0
   332.2      .1       0
Bank Sta=310.4,332.2
XS Rating Curve= 0 ,0
Exp/Cntr(USF)=0,0
Exp/Cntr=0.3,0.1

Type RM Length L Ch R = 1 ,37348   ,213.6,227,238.9
XS GIS Cut Line= 4
2439414.11538104636868.1830266752439553.60941887636740.206845183
2439638.07369865636645.504470878 2439762.2105947636489.373529458
#Sta/Elev= 30
       0 1954.25    17.1 1953.72    44.3 1949.68   98.031928.922   102.5 1927.46
   114.3 1928.15   125.9 1924.77   137.3 1922.88   158.3 1922.62   191.1 1920.75
   222.2 1916.87  229.431916.788   260.2 1914.54   269.1 1912.53     276 1911.98
   287.4 1912.28   293.31914.505   305.2 1924.32   318.5 1938.24   324.2 1943.43
     347 1963.72   355.5 1970.67   398.3 2000.81     432 2026.81   442.2 2033.57
   452.3 2041.02   462.6 2049.42   472.3 2055.44   500.7 2075.22   515.7 2084.45
#Mann= 5 ,-1 , 0
       0     .05       0   98.03     .06       0  229.43      .1       0
   260.2    .045       0   293.3      .1       0
Bank Sta=260.2,293.3
XS Rating Curve= 0 ,0
Exp/Cntr(USF)=0,0
Exp/Cntr=0.3,0.1

Type RM Length L Ch R = 1 ,37121   ,198.5,193.1,186.3
XS GIS Cut Line= 4
2439499.85942264636953.927068275 2439632.9546514636886.099692084
 2439702.0617894636880.9806448242439881.22844349 636695.41518166
#Sta/Elev= 30
       0  1952.1    40.1 1946.61      49 1944.67    60.9 1940.46    70.6 1935.23
      84 1926.88    97.5 1916.11   111.5 1913.53  124.371913.983   163.2 1913.91
   167.2  1913.3   173.61910.165   179.3 1908.26   191.3 1908.06   203.3  1909.1
   206.21910.152   211.3 1911.69  226.75  1912.4   248.5 1911.97   271.6 1913.37
     305  1913.6   317.6 1914.79   323.3 1915.93   338.3 1922.98   353.6  1927.4
   366.1 1935.64   375.1 1942.51   421.7 1982.81   466.2  2013.7   476.6 2020.22
#Mann= 5 ,-1 , 0
       0     .05       0  124.37     .06       0   173.6    .045       0
   206.2     .06       0  226.75      .1       0
#XS Ineff= 2 , 0
          133.32 1916.68
Permanent Ineff=
       F       F
Bank Sta=173.6,206.2
XS Rating Curve= 0 ,0
Exp/Cntr(USF)=0,0
Exp/Cntr=0.3,0.1

Type RM Length L Ch R = 1 ,36928   ,386.4,398,405.2
XS GIS Cut Line= 4
2439585.60346424637103.6592006212439681.58560036637085.742535212
2439737.89512022637055.0282516542439969.53200872636882.260406639
#Sta/Elev= 30
       0 1942.84    13.4 1938.15    29.1 1930.17    37.8 1924.69   57.761910.746
    62.2 1908.81    73.6 1906.98   103.5 1907.91   108.1 1907.72   114.11906.046
   121.7 1903.77   126.3 1903.43   135.4 1903.45     140 1904.88   141.5    1906
   144.5 1908.24   149.1 1910.18  160.671910.583   222.5 1908.92   247.7 1908.68
   257.7  1909.5   282.6 1908.16   317.5 1911.55   322.6 1913.37   331.1    1918
     354 1928.48   416.9 1963.95   432.3 1974.32   442.6 1977.15   450.8 1982.67
#Mann= 5 ,-1 , 0
       0     .05       0   57.76     .06       0   114.1    .045       0
   141.5     .06       0  160.67      .1       0
#XS Ineff= 2 , 0
                          161.67         1910.55
Permanent Ineff=
       F       F
Bank Sta=114.1,141.5
XS Rating Curve= 0 ,0
Exp/Cntr(USF)=0,0
Exp/Cntr=0.3,0.1

Type RM Length L Ch R = 1 ,36530   ,204.6,193.2,185.2
XS GIS Cut Line= 4
2439511.37727898637357.0520399762439833.87725634637403.123465313
2439920.90105975637424.8794161672440109.02604655637390.325847164
#Sta/Elev= 30
       0    1937    19.6 1933.18    78.8 1917.53    92.3 1915.24   104.4 1911.63
   116.5 1906.12   124.6 1903.58  179.741902.582   197.4 1904.09   229.7 1903.83
   286.2 1900.72   294.3 1902.58   314.5 1902.44   347.3 1901.03   351.4 1900.22
   354.2 1898.49   359.7 1896.42   363.8 1896.18   375.8 1896.76   379.51898.513
   384.4 1902.73  390.241910.853   392.6 1913.92   400.9 1920.24   421.4 1939.45
   473.7 1974.78  491.621985.393   521.8 2004.62   555.6 2024.52   606.7 2051.29
#Mann= 6 ,-1 , 0
       0     .05       0  179.74     .06       0   354.2    .045       0
   379.5     .06       0  390.24      .1       0  491.62      .1       0
#XS Ineff= 2 , 0
          201.02  1905.1
Permanent Ineff=
       F       F
Bank Sta=354.2,379.5
XS Rating Curve= 0 ,0
Exp/Cntr(USF)=0,0
Exp/Cntr=0.3,0.1

Type RM Length L Ch R = 1 ,36337   ,318.8,319.3,317.2
XS GIS Cut Line= 4
2439540.81180072637829.2841496832439817.24035274637646.278210149
2439945.21653424637575.8913103282440093.66890477637479.909174209
#Sta/Elev= 30
       0 1916.61    21.5 1909.69      32 1904.87    40.6 1901.79    59.9  1898.2
    81.1 1898.57   156.5 1897.89     229 1898.09   254.2 1897.54  347.711897.192
   410.8  1896.7   415.4 1896.38   420.91895.128   429.1  1892.6   438.2 1892.34
   444.1 1892.74   447.4 1893.67   449.8 1895.13  453.131897.531     463 1906.25
   471.3  1912.5   508.9  1939.4   517.5 1946.05  560.881976.985   569.9 1983.88
   579.4 1990.13     598 2000.73  612.452008.256   641.3  2024.7   654.4 2031.53
#Mann= 7 ,-1 , 0
       0     .05       0  347.71     .06       0   420.9    .045       0
   449.8     .06       0  453.13      .1       0  560.88      .1       0
  612.45      .1       0
#XS Ineff= 2 , 0
          139.32 1898.77
Permanent Ineff=
       F       F
Bank Sta=420.9,449.8
XS Rating Curve= 0 ,0
Exp/Cntr(USF)=0,0
Exp/Cntr=0.3,0.1

Type RM Length L Ch R = 1 ,36018   ,267.8,280.1,298.8
XS GIS Cut Line= 4
2439525.45465894638162.0222215632439995.12724502637909.909144023
2440068.07366847637862.5579568712440256.19865526 637703.86749182
#Sta/Elev= 30
       0 1916.84    33.2 1903.38    56.4 1900.38   119.5  1900.4   178.5 1898.69
   195.3 1897.06     233 1896.96   282.9 1895.28   296.6 1893.41   310.2 1893.71
   319.3 1892.06   345.9 1893.97   419.1 1894.14   437.5 1893.07   464.5 1893.45
  513.141891.938  539.311890.789   560.5 1890.04   566.8 1887.65   580.3 1887.47
   591.31890.045   595.7 1892.64   608.9 1904.12  621.081913.419   639.2 1928.57
   698.3 1966.64   726.7 1983.55   805.6 2026.51   840.3 2042.33   866.1 2055.24
#Mann= 6 ,-1 , 0
       0     .05       0  513.14    .055       0  539.31     .06       0
   560.5    .045       0   591.3     .06       0  621.08      .1       0
#XS Ineff= 2 , 0
           351.2 1893.83
Permanent Ineff=
       F       F
Bank Sta=560.5,591.3
XS Rating Curve= 0 ,0
Exp/Cntr(USF)=0,0
Exp/Cntr=0.5,0.3

Type RM Length L Ch R = 1 ,35738   ,50.1,65.2,70.4
XS GIS Cut Line= 4
2439531.82000512638204.7032573262440137.26910587638061.837097676
2440259.33888173638165.7946012772440462.86805623638109.039711294
#Sta/Elev= 30
       01924.327  15.335 1917.89  56.4331903.481  76.9831900.384  146.851899.623
 200.2781897.743 226.7271895.603 245.4871895.605 303.2071892.876 327.6841892.813
 352.3431891.542 359.7361890.073 368.7821889.668 381.1121891.603 504.4071891.422
 574.275 1888.95 648.3791886.996 666.888 1883.93 697.5711881.874 703.9041883.885
 708.0791887.188 714.6711889.484 760.6191888.238 782.4141889.155 790.7841893.952
 810.8661912.644 844.0871932.146 910.5291969.893 931.2921979.694 993.7092011.945
#Mann= 5 ,-1 , 0
       0     .05       0 574.275    .055       0 666.888    .045       0
 703.904    .055       0 844.087     .06       0
#XS Ineff= 2 , 0
          649.89 1888.78  714.89         1888.63
Permanent Ineff=
       F       F
Bank Sta=666.888,703.904
XS Rating Curve= 0 ,0
Exp/Cntr(USF)=0,0
Exp/Cntr=0.5,0.3

Type RM Length L Ch R = 1 ,35673   ,278.7,258.8,249
XS GIS Cut Line= 4
2439566.72009235638582.9248637422440139.15755217638114.148110935
2440264.70218621638245.4516731462440461.65752953638163.674893173
#Sta/Elev= 30
       0 1927.53    62.6  1922.8   132.6 1912.39   164.2 1910.06   195.8 1909.75
   397.8 1899.89   423.6  1897.8   457.7 1892.83   496.4 1892.86   517.7 1891.39
   542.9 1892.06   565.7 1890.29  591.56 1890.29  609.561890.391   650.3 1892.17
  706.371889.947   788.2 1886.01     7981883.639     808 1882.01   831.9 1880.93
   846.71883.641   855.1 1885.45  864.011885.406   958.7 1884.87   964.9 1887.36
  990.121905.881    1023 1930.39  1066.7 1957.45  1108.7 1977.68  1134.8 1991.69
#Mann= 8 ,-1 , 0
       0     .05       0  591.56     .06       0  609.56     .05       0
  706.37    .055       0     798    .045       0   846.7     .05       0
  864.01     .06       0  990.12      .1       0
Bank Sta=798,846.7
XS Rating Curve= 0 ,0
Exp/Cntr(USF)=0,0
Exp/Cntr=0.5,0.3

Type RM Length L Ch R = 1 ,35414   ,240.5,237.1,196.6
XS GIS Cut Line= 4
2439701.47901147638589.835577542 2440147.2200516638426.282017595
2440295.80039832638447.0141589972440531.91645317638276.549885249
#Sta/Elev= 30
       0 1934.47    26.9 1931.28    52.5 1926.77    99.3 1915.18   112.1 1910.56
   120.7 1909.87   133.4 1905.52   159.1 1902.09   180.3 1901.55   196.5 1899.01
   240.8 1898.01   355.5 1889.98   423.2 1888.38   457.3 1883.71   518.7 1883.11
   522.8 1882.57   526.61880.199   530.9 1878.13     543 1877.97     547 1877.98
   554.41880.232   623.8 1885.59   701.2 1882.51   746.9 1880.55   751.8 1881.47
   766.6 1894.27     789 1908.99  812.291921.787   870.5 1951.76     916 1970.73
#Mann= 5 ,-1 , 0
       0     .05       0   526.6    .045       0   554.4     .05       0
   701.2     .06       0  812.29      .1       0
#XS Ineff= 2 , 0
                          620.83         1885.74
Permanent Ineff=
       F       F
Bank Sta=526.6,554.4
XS Rating Curve= 0 ,0
Exp/Cntr(USF)=0,0
Exp/Cntr=0.5,0.3

Type RM Length L Ch R = 1 ,35177   ,41.7,41.2,43.8
XS GIS Cut Line= 4
2439793.62186214638752.2373518562440127.63969584638670.460571882
2440220.93433214638660.0945011822440590.65752047638445.862373363
#Sta/Elev= 30
       0 1966.27      30 1962.61    46.5 1959.47    75.3 1952.09    88.1 1947.79
   108.8 1943.02   132.9 1935.66   174.1  1921.2   202.9 1912.88   248.2 1895.77
   285.3 1884.37   314.1 1881.44   359.1 1878.76   371.2 1877.41   376.11875.927
   382.5 1873.86   391.3 1873.47   399.3 1873.59   407.3 1875.91   423.5 1877.01
   555.4 1878.57  701.89 1878.23   744.4 1878.79   767.8 1877.11   773.6 1877.53
   782.4 1880.69   800.4 1890.85   811.7 1896.18  839.021907.609   865.1    1918
#Mann= 5 ,-1 , 0
       0     .05       0   376.1    .045       0   407.3     .05       0
  701.89     .06       0  839.02      .1       0
#XS Ineff= 3 ,-1
       0     360 1876.86  421.25  701.38 1876.85  744.17  789.52  1879.1
Permanent Ineff=
       F       F       F
Bank Sta=376.1,407.3
XS Rating Curve= 0 ,0
Exp/Cntr(USF)=0,0
Exp/Cntr=0.5,0.3

Type RM Length L Ch R = 1 ,35136   ,163.6,158.9,147.8
XS GIS Cut Line= 4
2439787.86293397638846.6837737972440131.09505274638714.228425953
2440247.42540171638693.4962845512440606.78251934638476.960585466
#Sta/Elev= 30
       0 1982.63    42.3 1979.56      67 1976.67   122.7 1968.52   147.5  1963.6
     166 1958.02   183.2 1951.06     196    1947   217.5 1938.83   246.5  1926.6
   290.4  1911.5   343.8 1888.66   354.7 1884.57   367.9 1880.93   383.8 1878.06
   407.9 1875.54   416.3 1873.23   436.6 1872.84   445.41875.537   463.6 1876.47
   508.6 1876.89     616 1877.38   700.4 1876.56  760.611877.625   802.8  1877.6
   825.5 1875.91   834.2 1876.46     843 1879.07  867.621891.936   905.6 1907.45
#Mann= 5 ,-1 , 0
       0     .05       0   407.9    .045       0   445.4     .05       0
  760.61     .06       0  867.62      .1       0
Bank Sta=407.9,445.4
XS Rating Curve= 0 ,0
Exp/Cntr(USF)=0,0
Exp/Cntr=0.5,0.3

Type RM Length L Ch R = 1 ,34977   ,289.8,286,268.2
XS GIS Cut Line= 4
2439838.54150184639030.9694751462440217.47897524638866.264129566
2440391.39860589638777.5766357912440701.22894128 638558.73736544
#Sta/Elev= 30
       0 1997.99    26.4 1994.69   103.6 1980.42   170.5 1972.38   213.9 1963.66
   257.6 1951.56     323 1935.35   344.8    1928   388.4 1911.11   401.5 1900.12
   419.1 1887.33   423.6 1882.71   428.1 1876.28   431.61872.984   437.1  1870.8
   441.5 1870.69     455  1871.1     464 1872.97   504.4 1875.33   535.8 1875.76
   730.4 1873.09   784.9 1875.16   859.31874.286   891.6  1873.1   911.2 1875.75
   931.3 1875.62   945.5 1880.75     960 1883.56  969.83 1886.62   987.7 1893.06
#Mann= 5 ,-1 , 0
       0     .05       0   431.6    .045       0     464     .05       0
   859.3     .06       0  969.83      .1       0
Bank Sta=431.6,464
XS Rating Curve= 0 ,0
Exp/Cntr(USF)=0,0
Exp/Cntr=0.3,0.1

Type RM Length L Ch R = 1 ,34691   ,352,350.5,340.5
XS GIS Cut Line= 4
2440155.28255104639315.4605266042440355.69325126639132.326610888
2440423.64860363639060.9159016162440818.71107589638650.880216114
#Sta/Elev= 30
       0 1961.85    31.8 1953.71    70.8 1958.77    91.4 1957.77   127.4 1952.47
  176.111941.916   209.5 1935.22   223.7 1930.44   249.2 1919.16   264.8 1909.57
   294.5  1885.5   304.9 1874.79   315.4  1867.1   319.9 1865.12   331.2 1864.77
   339.5 1867.17   348.2 1869.48   391.8 1866.94  420.471868.188   450.1  1870.2
   535.9 1870.62   582.1 1869.09   717.3 1871.45   761.7 1870.69   789.5 1868.22
   872.8 1872.14   899.9 1876.91  911.961880.324   933.9 1880.98   939.4 1883.28
#Mann= 6 ,-1 , 0
       0    .055       0  176.11      .1       0   315.4    .045       0
   339.5      .1       0  420.47     .05       0  911.96     .06       0
#XS Ineff= 2 , 0
                          720.18         1871.76
Permanent Ineff=
       F       F
Bank Sta=315.4,339.5
XS Rating Curve= 0 ,0
Exp/Cntr(USF)=0,0
Exp/Cntr=0.3,0.1

Type RM Length L Ch R = 1 ,34340   ,377.3,376.2,367.6
XS GIS Cut Line= 4
  2440491.603956639525.0855118882440665.52358665 639314.30874097
2440801.43429139639123.1123258212440989.17534964638710.773069053
#Sta/Elev= 30
       0 2005.83    28.8 2000.65    67.8 1989.31   101.4 1984.06   136.9    1971
   163.6 1957.99   191.3 1941.63   220.7 1920.54   253.8 1895.51   285.2 1867.51
   293.31861.783     302 1859.24   311.8 1859.04   316.8 1859.35   323.8 1861.76
  331.311863.001   371.3 1863.94   414.3  1863.1     448 1864.59   480.3 1863.84
   508.1 1865.67   565.2  1866.4   644.3 1865.43   665.5 1864.29   735.5 1867.16
  821.451873.332   903.6 1878.92   919.7 1883.26   938.8 1884.27   960.9  1892.2
#Mann= 5 ,-1 , 0
       0      .1       0   293.3    .045       0   323.8      .1       0
  331.31     .05       0  821.45     .06       0
#XS Ineff= 2 , 0
                          586.21         1866.91
Permanent Ineff=
       F       F
Bank Sta=293.3,323.8
XS Rating Curve= 0 ,0
Exp/Cntr(USF)=0,0
Exp/Cntr=0.3,0.1

Type RM Length L Ch R = 1 ,33964   ,337.9,334.5,312.8
XS GIS Cut Line= 4
2440859.24318651639701.5251673452440984.05946229639513.510777251
2441187.87338096639165.9211485072441477.00475396638878.369728363
#Sta/Elev= 30
       0 1986.73      32 1968.64    46.4 1958.92   71.021948.101   142.4 1918.98
   171.8 1904.29   201.6 1887.17     231 1867.75   256.21854.925   270.3 1852.72
   279.7  1852.9   285.61854.883   294.2 1857.22  330.071858.975   363.2 1859.03
   386.4 1856.99   479.1 1858.68   507.8 1856.54  625.441860.842   660.9  1862.2
   723.3  1867.7   728.6 1868.81     735 1872.35  748.32 1873.78   762.4 1874.32
   773.7 1880.58   796.3 1889.46   931.7 1934.53   971.1  1950.3  1036.4 1973.03
#Mann= 7 ,-1 , 0
       0     .05       0   71.02      .1       0   256.2    .045       0
   285.6      .1       0  330.07     .05       0  625.44     .06       0
  748.32      .1       0
Bank Sta=256.2,285.6
XS Rating Curve= 0 ,0
Exp/Cntr(USF)=0,0
Exp/Cntr=0.3,0.1

Type RM Length L Ch R = 1 ,33629   ,289.1,282.7,270.9
XS GIS Cut Line= 4
2441127.83517239639802.6421502532441323.74932674639571.969032988
2441345.86866677 639513.510777252441630.63683924638968.108466849
#Sta/Elev= 30
       0 1931.45    25.9 1921.71    60.1 1911.11    84.8 1900.94   109.9 1888.65
   136.1 1873.44   172.2 1854.76   180.7 1852.76   200.5 1852.35     297 1852.53
   309.81850.899   316.6 1848.64   329.5 1848.01   351.51850.902   363.7 1852.65
   395.2 1852.41  413.461853.764   467.4 1854.67   489.3 1856.98     510 1857.37
     516 1859.51   527.8 1868.35  534.631871.138   557.5 1877.28   622.7 1898.07
  655.811905.098   729.4 1923.98     887 1973.89   922.1 1981.97   980.4 1998.42
#Mann= 7 ,-1 , 0
       0     .05       0   200.5      .1       0   309.8    .045       0
   351.5     .05       0  413.46     .06       0  534.63     .05       0
  655.81      .1       0
#XS Ineff= 2 , 0
                          427.24         1854.95
Permanent Ineff=
       F       F
Bank Sta=309.8,351.5
XS Rating Curve= 0 ,0
Exp/Cntr(USF)=0,0
Exp/Cntr=0.5,0.3

Type RM Length L Ch R = 1 ,33347   ,89,90,92.9
XS GIS Cut Line= 4
2441447.30350587 640191.025133522441612.24852905639732.026290938
2441580.30408457639613.2762909382441841.93602905639131.418652058
#Sta/Elev= 30
       0 1892.09    51.1  1896.9    85.2 1898.09   148.9  1892.1   196.7 1878.85
   259.4 1850.51   276.4 1846.11   327.4 1845.16   391.2 1847.04   420.9 1846.43
   549.5 1847.83   559.3 1846.42   567.6 1844.57   575.9 1844.31   588.3 1844.63
   600.5 1846.72   615.8 1850.91   640.7 1851.18   652.6 1859.53   666.1  1866.7
  740.631896.158  828.851929.678   863.8 1942.23     9031958.246     927 1966.09
   959.3 1980.31   980.1 1987.23  1038.8 2011.65    1102 2034.47    1159 2058.55
#Mann= 7 ,-1 , 0
       0     .05       0   549.5     .06       0   559.3    .045       0
   600.5     .06       0  740.63      .1       0  828.85      .1       0
     903      .1       0
#XS Ineff= 2 , 0
          529.96 1850.14     624            1850
Permanent Ineff=
       F       F
Bank Sta=559.3,600.5
XS Rating Curve= 0 ,0
Exp/Cntr(USF)=0,0
Exp/Cntr=0.5,0.3

Type RM Length L Ch R = 1 ,33257   ,238.6,248.1,258.3
XS GIS Cut Line= 4
2441519.01936239640195.6547631472441687.42214012639733.849207595
2441654.43602905639586.2797631472441883.60269567639162.668652043
#Sta/Elev= 30
       0  1886.7    43.4 1889.37    64.7  1888.9    84.6 1886.89   106.5 1880.78
   118.9 1874.36     186 1848.72   200.1 1845.94   311.6 1844.05   449.7 1845.35
  477.291846.963   506.9 1848.67   523.3 1848.55   531.5 1847.48   535.6 1845.66
   543.8  1843.5   556.1 1843.58  562.04 1845.73   568.5 1849.42  605.771862.157
   609.41863.198   633.9 1869.56     6461873.855   849.1 1958.55     862 1963.16
   952.4 2000.56   979.7 2010.22   996.7 2018.11  1088.2 2050.37  1124.4 2061.06
#Mann= 7 ,-1 , 0
       0     .05       0  477.29     .06       0   535.6    .045       0
  562.04     .06       0  605.77      .1       0   609.4     .06       0
     646      .1       0
Bank Sta=535.6,562.04
XS Rating Curve= 0 ,0
Exp/Cntr(USF)=0,0
Exp/Cntr=0.5,0.3

Type RM Length L Ch R = 1 ,33009   ,244.5,247.4,251
XS GIS Cut Line= 4
2441572.31797346640197.3908742822441836.90130681639853.640874267
2442059.81797346639576.5575409232442201.48464015639428.640874267
#Sta/Elev= 30
       0 1880.33    23.5 1879.71      32 1878.42    46.3 1873.44    73.8 1860.74
   111.9 1848.22   246.6 1841.74  384.351841.615   430.2  1843.3   462.3 1842.33
   488.7 1843.36   502.5  1842.8   519.31840.278   529.7 1839.83   543.7 1840.72
     548 1842.47   555.4 1847.75   579.3 1875.08   591.3 1885.24  652.491929.385
   673.2 1942.55   704.7  1964.9   736.6 1984.24   760.7 1998.08   793.6 2015.05
   829.4 2031.96     886 2050.91   934.1 2063.08   968.1 2069.38   994.2 2072.47
#Mann= 5 ,-1 , 0
       0     .05       0  384.35     .06       0   519.3    .045       0
   543.7      .1       0  652.49      .1       0
Bank Sta=519.3,543.7
XS Rating Curve= 0 ,0
Exp/Cntr(USF)=0,0
Exp/Cntr=0.3,0.1

Type RM Length L Ch R = 1 ,32761   ,286.7,288.9,287.6
XS GIS Cut Line= 4
2441557.58234972640287.6876776372442011.02881994639998.556304636
2442069.48707569639954.3176246142442243.28189006639813.701820258
#Sta/Elev= 30
       0 1872.49    20.4 1871.97    70.9 1866.77     101 1866.51   114.4 1863.18
     139 1859.15   153.2 1855.12   163.6 1853.42   290.8 1847.29   395.4 1839.23
  444.781837.745     528 1837.59   552.5 1839.51   557.3  1839.3   562.5 1838.05
   567.5 1836.73   572.5  1836.5   587.6 1836.62   593.41838.299     603 1844.11
  611.771850.746   628.6 1862.88   654.2 1880.08     677 1893.51   705.4 1912.94
   741.3 1933.79   753.8 1941.91  781.311955.282   792.8 1962.06   834.6 1980.45
#Mann= 6 ,-1 , 0
       0     .05       0  444.78     .06       0   562.5    .045       0
   593.4     .06       0  611.77      .1       0  781.31      .1       0
Bank Sta=562.5,593.4
XS Rating Curve= 0 ,0
Exp/Cntr(USF)=0,0
Exp/Cntr=0.3,0.1

Type RM Length L Ch R = 1 ,32472   ,84.5,86.6,90.6
XS GIS Cut Line= 4
2441696.61820121640387.2247076872442039.46797139640294.007489069
2442282.78071151640167.6112604342442443.93590302640058.594513237
#Sta/Elev= 30
       0 1860.07    14.6 1857.19      81 1856.08   118.3 1854.33   130.7 1851.18
   138.5 1850.75   155.6 1851.01   176.3 1849.54   213.6 1850.86     226 1849.35
   250.9 1843.55   275.7 1840.38   333.8 1838.13   368.9 1834.69   395.6 1833.44
   480.7 1832.74   523.2  1834.7  533.34 1832.62   539.3  1830.9   552.8 1831.09
  556.77 1832.62   566.3 1838.75   593.4 1859.59   629.5 1884.18   710.6 1929.82
   735.7 1941.02   740.5 1942.36   750.2  1942.9   798.5 1930.37     824 1926.61
#Mann= 5 ,-1 , 0
       0     .05       0   333.8      .1       0  533.34    .045       0
  556.77      .1       0     824     .05       0
Bank Sta=533.34,556.77
XS Rating Curve= 0 ,0
Exp/Cntr(USF)=0,0
Exp/Cntr=0.3,0.1

Type RM Length L Ch R = 1 ,32386   ,63,73.7,112.3
XS GIS Cut Line= 4
 2441743.1686637640406.4587758592442033.01921542640347.171163006
2442293.88471198640272.0735200582442471.74755054640162.720811906
#Sta/Elev= 30
       0 1865.02      69 1864.01   126.1 1861.35   183.3 1854.82   224.1 1843.78
   240.5 1841.21   260.9 1836.31   310.1  1834.3   326.8 1831.19   343.4 1830.91
   451.7 1831.09   479.2 1832.99   493.3 1832.86   497.71831.875   505.8 1829.88
     514 1829.84   518.3 1829.87   525.9 1831.77   530.2 1833.94   543.1 1843.59
   568.8 1858.29   587.1 1871.12   618.2 1890.09     624 1893.29   638.8 1899.42
   676.3 1910.22   699.8 1914.08   722.3 1913.14   742.1 1910.76   776.1  1905.3
#Mann= 4 ,-1 , 0
       0     .05       0   343.4      .1       0   497.7    .045       0
   525.9      .1       0
Bank Sta=497.7,525.9
XS Rating Curve= 0 ,0
Exp/Cntr(USF)=0,0
Exp/Cntr=0.5,0.3

Type RM Length L Ch R = 1 ,32312   ,92.4,104.2,87.5
XS GIS Cut Line= 4
2441750.33659838640418.823764845  2442231.820219640335.524741947
 2442302.7241426640423.7981501872442537.45496157640596.378059091
#Sta/Elev= 30
       01869.091  69.9991866.964 126.2571864.139  174.97 1855.25 191.2071851.432
 211.5041843.949 231.8021838.001  239.921836.714 256.1581835.273 276.455 1834.95
 325.1681830.555 426.6541829.506 446.9511830.469 474.4111833.303 507.3371830.789
 515.8731829.187 544.3251828.781 557.1811829.231 564.241 1830.75 576.3431832.107
 590.4351832.076 607.0811829.974 641.6041830.768 651.5331832.938 656.4981835.161
 678.477 1833.27 694.8661836.986 729.9781839.606 816.4151875.003 893.2051905.244
#Mann= 4 ,-1 , 0
       0     .05       0 426.654      .1       0 507.337    .045       0
 564.241      .1       0
#XS Ineff= 2 , 0
          453.25 1833.86  616.59         1833.82
Permanent Ineff=
       F       F
Bank Sta=507.337,564.241
XS Rating Curve= 0 ,0
Exp/Cntr(USF)=0,0
Exp/Cntr=0.5,0.3

Type RM Length L Ch R = 1 ,32208   ,91,87.6,83.2
XS GIS Cut Line= 4
2441765.74903851640471.4466859012442226.62454188640432.262938652
2442304.05909001640546.0823949482442528.89916351640660.834797606
#Sta/Elev= 30
       0 1886.23   33.861881.116    56.9 1877.27    73.3  1876.9   129.5 1866.19
   161.6 1856.48   213.8 1835.58   225.8 1832.95     270 1832.05     286 1828.88
   298.1 1828.14   341.8 1829.08   394.4 1828.15  432.271830.577   462.5 1832.78
   469.9 1828.65   499.6 1827.03   507.7 1828.74   513.5 1832.82   519.2 1834.41
  560.471833.068  613.74    1834   675.1 1834.82   681.2 1835.93   705.4 1844.92
  736.891856.904   748.5 1860.57   773.9 1871.89   796.3 1880.37   852.6 1900.28
#Mann= 9 ,-1 , 0
       0      .1       0   33.86     .05       0  432.27     .06       0
   469.9    .045       0   507.7     .06       0  560.47     .05       0
  613.74     .06       0   705.4    .055       0  736.89      .1       0
Bank Sta=469.9,507.7
XS Rating Curve= 0 ,0
Exp/Cntr(USF)=0,0
Exp/Cntr=0.5,0.3

Type RM Length L Ch R = 1 ,32120   ,184.6,178.3,168
XS GIS Cut Line= 4
2441788.13975123640481.7090958952442163.18418919640493.837398615
2442206.09972189640544.2165022212442487.84952354640693.487920314
#Sta/Elev= 30
       0 1886.76   13.551884.451    42.6 1878.94    58.6 1878.14    66.6  1875.5
   118.7 1864.44   139.4 1858.29   190.7 1839.16   210.7 1833.42   262.7 1827.05
   329.3  1827.5   348.7 1826.62   378.5 1827.97   386.9    1827   398.4    1825
   408.2 1825.22   414.71827.475   418.7  1830.2   423.9 1831.47   488.3 1827.55
   500.1 1828.04   528.2 1831.58  572.671832.516  576.011832.563   614.2 1831.54
   641.3 1832.08   677.5 1844.37  700.571853.578   731.9 1864.61   760.3 1877.09
#Mann= 7 ,-1 , 0
       0      .1       0   13.55     .05       0   386.9    .045       0
   414.7     .05       0  572.67    .035       0  576.01    .055       0
  700.57      .1       0
#XS Ineff= 2 , 0
                          423.75         1831.43
Permanent Ineff=
       F       F
Bank Sta=386.9,414.7
XS Rating Curve= 0 ,0
Exp/Cntr(USF)=0,0
Exp/Cntr=0.3,0.1

Type RM Length L Ch R = 1 ,31942   ,125.8,118.2,95.9
XS GIS Cut Line= 4
2441799.33510758640625.3828358092442016.71161018640621.651050357
2442096.01205104640656.170065791 2442435.6045272640687.890242136
#Sta/Elev= 30
       0  1908.1    15.4 1903.93    43.4 1894.88    51.4 1891.09    63.4 1889.45
    71.4 1886.07  125.861869.972   167.1 1853.56   187.4 1844.94   211.4 1833.63
  227.761827.344   237.1 1825.13     2461824.913   253.3 1823.23   267.6 1822.61
   274.6 1822.94   280.6 1824.67   289.8 1827.06   308.9 1825.02   322.7 1824.96
  340.331823.179  442.941824.695   499.5 1823.09   507.5    1826   523.6 1829.85
  545.541830.845   605.2 1829.98   607.9 1830.56     620 1838.32     645  1850.4
#Mann= 8 ,-1 , 0
       0      .1       0  125.86     .05       0  227.76      .1       0
     246    .045       0   280.6      .1       0  340.33     .05       0
  442.94    .035       0  545.54    .055       0
#XS Ineff= 2 , 0
                          461.94         1829.04
Permanent Ineff=
       F       F
Bank Sta=246,280.6
XS Rating Curve= 0 ,0
Exp/Cntr(USF)=0,0
Exp/Cntr=0.3,0.1

Type RM Length L Ch R = 1 ,31824   ,175.3,174,168.2
XS GIS Cut Line= 4
2441853.44599664640789.5813957112442017.64455654640757.861219367
2442087.61553378640750.3976484622442446.79988356640700.018544856
#Sta/Elev= 30
       0 1910.93    13.5  1906.1    21.7 1901.52    33.9 1899.18    74.7 1879.64
   111.3 1866.84   143.9 1853.17   168.3  1840.3   180.4 1831.95   190.91823.162
   196.5 1820.91   204.5 1820.76   212.6 1821.37   216.6 1822.57   241.9 1824.76
   268.3  1825.1  296.251822.642   349.7 1824.31   386.2 1823.74  395.591824.404
   406.4 1824.94   458.9 1823.15   463.1  1823.6   479.1 1828.61  494.931830.025
   555.8 1829.27   559.9  1830.8     572 1839.03  594.271850.629   600.3 1853.87
#Mann= 7 ,-1 , 0
       0      .1       0   190.9    .045       0   216.6      .1       0
  296.25    .055       0  395.59    .035       0  494.93    .055       0
  594.27      .1       0
#XS Ineff= 2 , 0
                          411.22         1827.55
Permanent Ineff=
       F       F
Bank Sta=190.9,216.6
XS Rating Curve= 0 ,0
Exp/Cntr(USF)=0,0
Exp/Cntr=0.3,0.1

Type RM Length L Ch R = 1 ,31650   ,225.5,224.7,225.2
XS GIS Cut Line= 4
2441886.09911935640950.0481701612442027.90696654640933.255135626
2442396.42077996640863.2841583952442472.92238173640845.558177496
#Sta/Elev= 30
       0 1914.04     8.7 1909.01    20.8 1906.13      49 1894.06    86.3 1874.36
   117.5    1854   122.3 1849.97   133.6 1838.33   159.51820.754     166 1818.47
   186.4 1818.65   194.5 1820.48   198.6 1822.19   202.7 1822.79   214.9 1820.83
   239.3 1819.91  289.691820.621   308.1 1820.59   328.9 1823.01  389.051824.051
   434.9 1824.47   491.8 1822.38     504 1825.46   516.2 1826.82   528.5 1826.66
   553.1  1824.5   573.7    1825   577.8 1825.49  587.881830.795   596.4 1834.59
#Mann= 6 ,-1 , 0
       0      .1       0   159.5    .045       0   194.5      .1       0
  289.69    .055       0  389.05    .035       0  587.88      .1       0
#XS Ineff= 2 , 0
                          392.86         1824.43
Permanent Ineff=
       F       F
Bank Sta=159.5,194.5
XS Rating Curve= 0 ,0
Exp/Cntr(USF)=0,0
Exp/Cntr=0.3,0.1

Type RM Length L Ch R = 1 ,31425   ,262.8,260.3,227.5
XS GIS Cut Line= 4
2441922.48402751641153.4304773122442033.50464472641163.692887306
2442379.62774542641081.5936073552442576.47942803641021.885040118
#Sta/Elev= 30
       0 1892.65    44.4 1878.32    84.6 1861.92    97.2 1853.51   108.7 1847.14
   133.1 1836.87   149.7  1828.3   157.71818.268   162.1 1816.55   182.7 1815.84
   190.9 1816.46     195 1818.38   199.1  1820.1   211.4 1817.88   227.9 1817.31
   264.9  1817.8     276 1816.99  290.161818.405  358.571818.786   372.4 1822.01
   392.3 1823.06   449.9 1822.42   487.2 1824.06   531.7 1823.94   545.7 1821.88
   566.6 1823.03  589.66 1821.49   612.6  1822.2   641.8  1839.7   672.9 1855.96
#Mann= 6 ,-1 , 0
       0      .1       0   157.7    .045       0     195      .1       0
  290.16     .06       0  358.57    .035       0  589.66     .06       0
#XS Ineff= 2 , 0
                          317.16         1821.65
Permanent Ineff=
       F       F
Bank Sta=157.7,195
XS Rating Curve= 0 ,0
Exp/Cntr(USF)=0,0
Exp/Cntr=0.3,0.1

Type RM Length L Ch R = 1 ,31165   ,287.6,284.7,238.6
XS GIS Cut Line= 4
2442014.84571746641464.101616218 2442132.3969592641410.923673522
2442558.75344713641212.2060981862442659.51165434641167.424672758
#Sta/Elev= 30
       0 1902.91    30.6 1888.64    39.4 1883.73    48.2 1880.84      57 1875.54
    65.7 1872.18    82.5 1862.58   100.6 1851.34     114 1841.95   131.6 1831.58
   138.6 1825.47   147.51814.728   149.3 1813.06   151.9 1812.35   158.1 1812.03
   166.9 1812.37     173 1814.74   184.6 1817.33   223.8 1814.67  253.87 1814.98
   312.5    1816   325.8 1817.95   356.6  1817.6   378.7 1816.79  563.491817.608
   599.4  1817.1     630 1819.47   639.8 1825.31  666.371838.226   709.7 1863.26
#Mann= 7 ,-1 , 0
       0      .1       0   147.5    .045       0     173      .1       0
  253.87    .055       0   356.6      .1       0  563.49     .06       0
  666.37      .1       0
#XS Ineff= 2 ,-1
  328.11  547.281817.792  557.41  638.46 1819.03
Permanent Ineff=
       F       F
Bank Sta=147.5,173
XS Rating Curve= 0 ,0
Exp/Cntr(USF)=0,0
Exp/Cntr=0.3,0.1

Type RM Length L Ch R = 1 ,30880   ,263,251.6,230.8
XS GIS Cut Line= 4
2442135.19579829641747.7173105942442276.07069912641667.483923369
2442503.70961171641487.4252752952442748.14155884641359.611623553
#Sta/Elev= 30
       0  1862.3      34 1854.55    90.6 1845.65   122.9 1837.88   155.7 1833.66
   170.1 1827.73   180.8 1818.98   185.9 1815.73     191 1813.72   206.3 1812.03
   216.9 1811.82   231.8 1809.95   257.3 1809.63   285.6    1812  298.021812.485
   308.3 1811.22   321.1 1810.77   382.3 1812.77   426.4 1813.35   440.9  1814.4
     519 1814.66   594.3 1813.77  624.281814.447   635.8 1815.29   649.9  1815.2
   653.6 1816.18   663.4 1824.04     677 1831.11   689.2 1838.72   728.2 1865.28
#Mann= 5 ,-1 , 0
       0      .1       0   216.9    .045       0   285.6      .1       0
  298.02     .05       0  624.28     .06       0
#XS Ineff= 2 , 0
                          469.62         1814.62
Permanent Ineff=
       F       F
Bank Sta=216.9,285.6
XS Rating Curve= 0 ,0
Exp/Cntr(USF)=0,0
Exp/Cntr=0.3,0.1

Type RM Length L Ch R = 1 ,30628   ,371.3,367,345.2
XS GIS Cut Line= 4
2442278.86953821641882.0615868772442520.50264625641752.382042409
2442600.73603347641705.7347242552442860.09512241641566.725716156
#Sta/Elev= 30
       0 1898.61    27.1 1884.67    58.9 1863.48    90.7 1844.65    99.7 1838.22
   114.5 1825.62   126.3 1817.42     136  1812.3   145.1 1808.98   149.7 1808.25
   172.4  1807.3   226.8 1807.94   235.9  1808.7   247.4 1807.55     300    1808
   309.1 1807.16   320.9 1808.22   332.9 1809.35  370.191809.457  475.221809.598
   528.2 1809.84   546.3 1810.91   556.8 1812.53   576.3 1813.15   578.1 1813.46
  580.241814.958   587.2 1820.36   609.9 1831.18   641.6 1850.48   661.3 1859.97
#Mann= 6 ,-1 , 0
       0      .1       0     300    .045       0   320.9      .1       0
  370.19     .05       0  475.22     .06       0  580.24      .1       0
Bank Sta=300,320.9
XS Rating Curve= 0 ,0
Exp/Cntr(USF)=0,0
Exp/Cntr=0.3,0.1

Type RM Length L Ch R = 1 ,30261   ,399.5,401.2,376
XS GIS Cut Line= 4
 2442412.1317481642179.2788149322442591.29840219642102.493106037
2442949.63171037641910.5288337982443105.76265179641824.784792198
#Sta/Elev= 30
       0 1920.12    15.9 1914.06    69.3 1898.61    85.5 1892.65   107.3 1878.38
   124.1 1862.71   154.6 1839.47     182 1820.51     206 1805.87   219.21802.723
   253.4 1800.53   273.51802.715   285.1 1804.58   339.5 1803.32  380.09 1804.06
     453  1803.9  485.111804.994   561.9 1804.21   575.5 1806.79   593.6 1807.94
   598.2 1809.48   607.3 1816.22   625.6 1824.26   634.4  1829.9   643.8 1833.53
   660.81844.432   671.2 1849.64   698.5 1866.73   713.9 1875.23   779.6 1908.97
#Mann= 6 ,-1 , 0
       0      .1       0   219.2    .045       0   273.5      .1       0
  380.09     .05       0  485.11     .06       0   660.8      .1       0
Bank Sta=219.2,273.5
XS Rating Curve= 0 ,0
Exp/Cntr(USF)=0,0
Exp/Cntr=0.3,0.1

Type RM Length L Ch R = 1 ,29860   ,395,396.7,386.6
XS GIS Cut Line= 4
2442633.53054209642517.1359340722442776.86386536642444.189510621
2443132.63764991642224.0704784552443223.50073877642114.010962371
#Sta/Elev= 30
       0 1892.55    46.2 1876.89    95.6 1853.47   133.4 1837.01   142.4 1832.27
   158.5 1821.85   190.41797.879     198 1795.72     212 1795.24   219.5 1795.35
   227.31797.868   231.7 1798.86   246.9 1799.53  318.831799.374   355.9 1798.55
   389.8 1799.39   468.3 1799.29  533.881800.221   555.4 1801.35   558.3 1802.09
     567 1806.33   584.4 1807.93   587.2 1808.76   595.7 1814.55   621.3 1827.27
  655.631846.156   663.9 1850.49   694.8 1864.17   710.4 1870.29   721.9 1876.13
#Mann= 6 ,-1 , 0
       0      .1       0   190.4    .045       0   227.3      .1       0
  318.83     .05       0  533.88     .06       0  655.63      .1       0
Bank Sta=190.4,227.3
XS Rating Curve= 0 ,0
Exp/Cntr(USF)=0,0
Exp/Cntr=0.3,0.1

Type RM Length L Ch R = 1 ,29464   ,465.8,466.4,357.7
XS GIS Cut Line= 4
2442899.72099959642816.6001987642442999.54242115642764.129964352
2443345.07811118642538.8918849262443485.85191083642451.868081511
#Sta/Elev= 30
       0 1846.92      35 1835.78    57.6 1827.07    89.3  1812.5   138.2 1792.84
   144.9 1791.09   156.4 1790.43   162.2 1790.71   173.9 1792.83   182.5 1793.89
     193 1794.12   283.7 1792.09  305.231792.249  413.851795.531   465.2 1796.21
   477.3 1797.99     486 1796.01   497.5    1799   514.9 1799.62   517.8 1800.47
   526.4 1807.78   532.8 1812.02   555.7 1822.72  574.391832.904   608.9 1850.27
   630.7 1858.89   642.7 1866.67   648.5 1869.57   668.8 1875.72   690.7 1880.82
#Mann= 6 ,-1 , 0
       0      .1       0   138.2    .045       0   173.9      .1       0
  305.23     .05       0  413.85     .06       0  574.39      .1       0
Bank Sta=138.2,173.9
XS Rating Curve= 0 ,0
Exp/Cntr(USF)=0,0
Exp/Cntr=0.3,0.1

Type RM Length L Ch R = 1 ,28997   ,394.6,399.7,399
XS GIS Cut Line= 4
2443090.40551001643132.7013670512443425.70310552 642885.70733677
2443488.41143446642828.1180550992443634.30428136642665.588304603
#Sta/Elev= 30
       0  1830.4    35.9 1816.16    93.1 1791.18     111  1788.8  163.281787.948
   196.1 1787.36   253.8 1788.76  381.991787.298  386.541787.804     401  1788.4
   427.81786.711   436.2 1784.46   444.7 1784.07   456.1 1784.11   462.31786.733
   470.1 1793.11   477.6 1796.82   498.4 1798.59   501.3 1801.93   506.9 1810.69
   512.6 1816.07     529 1826.96  555.821841.445     565 1846.51   608.9 1875.26
   628.7 1885.09   637.6  1888.3   666.8 1894.16   705.2 1905.14     720 1908.14
#Mann= 7 ,-1 , 0
       0      .1       0  163.28     .05       0  381.99      .1       0
  386.54     .06       0   427.8    .045       0   462.3     .06       0
  555.82      .1       0
Bank Sta=427.8,462.3
XS Rating Curve= 0 ,0
Exp/Cntr(USF)=0,0
Exp/Cntr=0.3,0.1

Type RM Length L Ch R = 1 ,28597   ,771.8,773.3,773.1
XS GIS Cut Line= 4
2443246.53645144643476.9572952652443561.35785791643264.516833988
2443720.04832296 643142.939461572443864.66140804643012.403756448
#Sta/Elev= 30
       0 1816.35    53.3 1800.74    87.1 1791.58   106.4 1787.41  124.871784.448
   140.2 1783.28   191.8 1782.47   260.8    1782   344.5 1782.46   382.5 1781.44
   447.6 1782.83   454.8 1781.65   461.8 1779.07   467.2 1778.65   473.2 1779.01
   482.61781.511   494.3    1783   546.9 1783.08   553.5 1783.76  560.551786.505
   564.5 1788.34     573 1790.05   597.7 1790.73   618.5 1800.43   655.3 1814.03
   669.4 1818.38   712.7 1829.29  724.081831.457   762.9  1841.2   774.5 1843.47
#Mann= 6 ,-1 , 0
       0      .1       0  124.87     .05       0   454.8    .045       0
   482.6     .05       0  560.55     .06       0  724.08      .1       0
Bank Sta=454.8,482.6
XS Rating Curve= 0 ,0
Exp/Cntr(USF)=0,0
Exp/Cntr=0.3,0.1

Type RM Length L Ch R = 1 ,27824   ,464.8,467.3,465.1
XS GIS Cut Line= 4
2443547.24679829644127.0542992742443783.48117622644007.853466371
2444271.12094719643678.4257099852444451.00584048643580.897755792
#Sta/Elev= 30
       0 1794.63    62.3    1788   133.8 1783.08   172.5 1776.45   201.1 1774.37
   331.3  1774.4   446.3 1772.55   538.9 1773.38   601.6 1771.97   645.1 1772.16
     674 1773.76   680.51771.705   688.5 1768.94   702.7 1769.13   718.21771.696
   736.8 1773.96   770.6 1775.21  810.061780.789   832.3 1785.34   846.7 1795.16
   852.6 1797.17     882 1798.73   887.9 1802.18   902.6 1815.43  916.931820.399
   957.3 1828.32   975.5 1834.19   994.1 1842.76  1030.1 1863.78  1057.7 1875.06
#Mann= 5 ,-1 , 0
       0     .05       0   680.5    .045       0   718.2      .1       0
  810.06     .06       0  916.93      .1       0
Bank Sta=680.5,718.2
XS Rating Curve= 0 ,0
Exp/Cntr(USF)=0,0
Exp/Cntr=0.3,0.1

Type RM Length L Ch R = 1 ,27357   ,229.9,241.4,230.7
XS GIS Cut Line= 4
2443564.58510126644163.8981930812444227.77518977644224.582253468
2444626.55615803644001.3516027592444719.74953648 643847.47416392
#Sta/Elev= 30
       0 1790.63    26.3 1788.27   126.7 1783.21   170.9 1782.45   231.1 1779.77
   399.61777.362  452.421775.436   480.2  1775.7   568.5 1770.76  657.531769.857
   793.1 1767.09   848.1 1766.95  868.691765.284   882.3 1765.15   903.2 1763.89
   913.3 1764.99   922.1 1769.01   939.7 1765.75   971.9 1765.81  1046.1 1768.42
  1060.3 1769.72 1080.11 1773.77  1110.2 1780.76  1123.3 1785.93  1148.2 1786.99
  1165.7 1790.54  1186.6  1799.4 1214.051807.251 1254.091816.725  1302.9 1830.66
#Mann= 10 ,-1 , 0
       0     .06       0   399.6     .05       0  452.42     .06       0
  657.53     .05       0  868.69      .1       0   882.3    .045       0
   913.3      .1       0 1080.11     .06       0 1214.05      .1       0
 1254.09      .1       0
Bank Sta=882.3,913.3
XS Rating Curve= 0 ,0
Exp/Cntr(USF)=0,0
Exp/Cntr=0.5,0.3

Type RM Length L Ch R = 1 ,27115   ,64.3,62.7,70
XS GIS Cut Line= 4
2443878.56797346644305.7242075952444372.31797346 644324.47420761
2444520.23464012644332.8075409232444899.40130681 644055.72420761
#Sta/Elev= 30
       0 1774.06       9 1773.76    44.2 1779.59    96.2 1781.92   140.3 1778.03
   160.3  1774.4  255.231772.295   380.5 1767.43   410.9 1764.48   427.5 1766.24
   532.6 1764.06   560.6 1762.96   564.6 1761.41   572.7  1760.3   587.5 1761.48
   596.7 1761.62   608.7 1764.22   624.7 1761.94   731.3 1764.57   794.7 1767.15
   853.4 1771.96   869.2 1771.71   907.9 1775.31   928.8  1781.7     966 1783.44
  997.151786.604  1026.1 1795.21  1081.3 1808.25 1108.571810.177  1111.9 1810.37
#Mann= 6 ,-1 , 0
       0     .05       0  255.23     .06       0   564.6    .045       0
   587.5     .06       0  997.15      .1       0 1108.57     .12       0
#XS Ineff= 2 , 0
          427.36 1766.33     615         1761.88
Permanent Ineff=
       F       F
Bank Sta=564.6,587.5
XS Rating Curve= 0 ,0
Exp/Cntr(USF)=0,0
Exp/Cntr=0.5,0.3
